HEC-RAS study lds_broad_rvr.prj: Upper_Broad 3-06-07

--- lds_broad_rvr.g05 (geometry) --- (continued)

Type RM Length L Ch R = 1 ,387269.9,68.66,91.62,104.15
XS GIS Cut Line= 6
 1033627.0796561  660907.7254103  1033573.249208  660879.5679582
 1033535.9049101  660875.5215836 1033488.8388405  660879.8003254
 1033445.1007047  660863.6362265 1033391.0538708  660863.8329078
#Sta/Elev= 30
       0 2195.66    5.18 2194.35    9.77 2192.88   22.31 2190.49   35.55 2188.55
   41.35 2188.22   48.14 2184.37   52.84 2182.78   66.56 2182.26    79.4 2179.25
   89.77 2178.12   98.47 2173.73  111.65 2168.41  118.14 2166.17  128.86 2166.31
  134.81 2167.11  142.17 2166.56  146.92 2167.61  153.79 2170.21  166.19 2173.82
  167.87 2174.95  178.93 2179.96  179.79 2179.95   184.3 2180.79  193.07 2181.37
  200.03 2181.53  227.73 2181.34   231.7 2181.99  236.39  2186.9   248.1 2199.87
#Mann= 3 , 0 , 0
       0     .08       0  111.65     .05       0  153.79    .065       0
Bank Sta=111.65,153.79
Exp/Cntr=0.3,0.1

Type RM Length L Ch R = 1 ,387178.3,101.19,89.51,82.3
XS GIS Cut Line= 6
 1033645.2991928  660843.1288847 1033622.1106833  660816.6277266
 1033563.3112926  660814.1432704 1033461.4475314  660751.2030388
 1033401.8199483   660752.031201 1033373.6624962  660761.9691466
#Sta/Elev= 30
       0  2193.4    4.99 2192.51   17.53 2188.93   19.22 2188.84    26.2  2187.2
   34.23 2186.26   40.23 2185.01   60.45 2182.44   89.75  2180.2   95.12 2178.81
   97.36  2177.3  106.74 2172.64  109.47 2171.74  115.76 2168.48  127.93 2164.65
   130.8 2164.27  137.63 2164.89  154.58 2165.56  162.52 2168.96  177.79  2176.3
  194.56 2181.01  204.22 2181.25  234.69 2180.68  264.17 2179.51  269.03 2178.96
  276.53 2179.01  278.64 2181.18   291.5  2198.7  298.86 2204.71   303.3 2208.93
#Mann= 3 , 0 , 0
       0     .08       0  115.76     .05       0  162.52    .065       0
Bank Sta=115.76,162.52
Exp/Cntr=0.5,0.3

Type RM Length L Ch R = 1 ,387088.8,14.98,17.54,19.94
XS GIS Cut Line= 6
 1033730.5997416  660713.9358335 1033598.8247108  660727.4788769
 1033538.8688413   660696.644434 1033520.0255723  660693.2183713
 1033449.0250993  660719.7329382 1033372.8343341  660723.8737488
#Sta/Elev= 30
       0 2187.26    2.27 2186.81   18.53 2186.02   36.65 2183.74   51.55 2182.51
   70.58 2180.12   94.33 2177.54  101.99 2176.91  106.63 2177.07  119.99 2174.53
  121.97 2173.74  128.75 2172.99  132.26 2172.26  134.22 2171.74  143.36  2168.1
  150.74 2166.07  155.01 2164.98  163.28 2163.71  172.12 2163.68  188.31 2164.34
   199.1 2167.15  229.76 2178.54  233.78 2179.24  248.84 2180.49  262.46 2181.38
  314.86 2180.19  348.57 2178.34  351.44 2179.94  366.98 2192.63  371.42 2196.74
#Mann= 3 , 0 , 0
       0     .08       0  150.74     .05       0   199.1    .065       0
Bank Sta=150.74,199.1
Exp/Cntr=0.5,0.3

Type RM Length L Ch R = 3 ,387080. ,,,
BEGIN DESCRIPTION:
STR_153
END DESCRIPTION:
Bridge Culvert--1,0,-1,-1, 0
Deck Dist Width WeirC Skew NumUp NumDn MinLoCord MaxHiCord MaxSubmerge Is_Ogee
2,12,2.6,0, 2, 2, 2175, , 0.95, 0, 0,0,,
       0     260
    2175    2175
    2174    2174
       0     260
    2175    2175
    2174    2174
Pier Skew, UpSta & Num, DnSta & Num=  ,145, 2 ,106, 2 , 0 , 0 , 0 ,,
       1       1
    2160    2174
       1       1
    2160    2174
Pier Skew, UpSta & Num, DnSta & Num=  ,165, 2 ,126, 2 , 0 , 0 , 0 ,,
       1       1
    2160    2174
       1       1
    2160    2174
Pier Skew, UpSta & Num, DnSta & Num=  ,185, 2 ,146, 2 , 0 , 0 , 0 ,,
       1       1
    2160    2174
       1       1
    2160    2174
Pier Skew, UpSta & Num, DnSta & Num=  ,205, 2 ,166, 2 , 0 , 0 , 0 ,,
       1       1
    2160    2174
       1       1
    2160    2174
BR Coef=-1 , 1 , 0 ,, 0 ,,,0.8,0,2,0,
WSPro=,,,, 1 ,,,, 0 ,,,, 0 ,,,,-1 ,-1 ,-1 , 0 , 0 , 0 , 0 , 0
BC Design=,, 0 ,, 0 ,,,,,,

Type RM Length L Ch R = 1 ,387071.2,118.36,122.23,79.06
XS GIS Cut Line= 6
 1033685.8790467  660694.8881346 1033623.6635819   660715.487703
  1033600.537727  660711.2051473 1033528.5907138  660674.3751024
 1033461.4475314  660687.4346754 1033357.9274459  660700.6852393
#Sta/Elev= 30
       0 2183.05   11.33 2182.26   49.04    2178   56.59 2176.91   73.78 2175.75
   82.72 2174.83   90.46 2170.87   99.25 2164.58  105.74 2163.26  122.96 2163.15
  137.59 2163.44  143.66 2165.85  166.67 2173.44  168.13 2174.08  170.69 2174.21
  178.09 2175.79  187.17 2177.01  190.91 2177.78  199.51 2178.94  201.78 2179.53
  210.76 2180.75  237.34  2181.2  265.17 2180.52  279.72 2179.95  294.93 2178.94
  310.23 2177.86  318.49 2176.97  333.46 2191.28  341.17 2200.22  342.95  2201.6
#Mann= 3 , 0 , 0
       0     .08       0   99.25     .05       0  143.66    .065       0
Bank Sta=99.25,143.66
Exp/Cntr=0.5,0.3

Type RM Length L Ch R = 1 ,386949.0,421.12,314.21,145.31
XS GIS Cut Line= 6
  1033706.745276  660650.3927546 1033676.7673261  660620.4148349
 1033616.8114868  660580.1587576 1033577.4119024  660572.4501393
  1033504.608366  660610.9932005 1033458.3566866  660664.9534679
#Sta/Elev= 30
       0 2183.27    8.68  2182.4   11.36 2182.93   43.15 2177.12   49.56 2176.86
   60.61 2176.02   72.73 2170.72   87.93 2165.59   92.54 2164.27  102.61 2162.67
  114.84 2160.99  117.97 2160.35  120.06 2160.36  127.13  2161.2  142.48 2163.87
  154.99 2166.17  173.58 2167.53  195.61 2171.67  198.67 2171.65  206.07  2172.1
  215.11 2172.38  233.03 2173.79  237.81 2174.54  250.82 2177.85  256.89 2178.15
  261.37 2178.61  266.17 2179.36  279.43 2180.11  303.15 2181.02  308.68 2181.09
#Mann= 3 , 0 , 0
       0      .1       0  102.61     .05       0  142.48    .065       0
Bank Sta=102.61,142.48
Exp/Cntr=0.3,0.1

Type RM Length L Ch R = 1 ,386634.8,212.29,213.54,231.39
XS GIS Cut Line= 6
 1033438.6670947  660347.3484909 1033437.3310964  660406.1327476
 1033445.3471163  660424.8368141 1033434.6590696   660496.981114
 1033445.3471163   660550.421317 1033447.3687751   660637.745038
#Sta/Elev= 30
       0 2191.05    1.38 2190.64      29 2158.63   31.08 2155.99   46.13 2156.21
   48.66 2156.09   61.05 2157.09   63.12 2157.25   75.35 2158.64   77.13 2159.54
    79.8 2160.16   93.21 2165.36    94.5 2165.53   97.03 2166.12  111.81 2167.19
  120.19 2167.41  143.73 2167.45  147.05  2167.6  152.16 2167.43  164.06 2167.32
  187.82  2168.5     191  2168.8  198.71 2169.17  227.08 2171.91  242.43 2174.13
  252.11 2175.38   255.2 2175.95  268.27 2177.61  282.91 2179.22  294.21 2180.12
#Mann= 3 , 0 , 0
       0      .1       0      29     .05       0   61.05    .065       0
Bank Sta=29,61.05
Exp/Cntr=0.3,0.1

Type RM Length L Ch R = 1 ,386421.3,177.15,187.32,211.86
XS GIS Cut Line= 6
 1033262.3143853   660367.388586 1033231.5862738   660432.852834
 1033222.2342254  660479.6130154 1033192.8421122  660504.9971338
 1033190.1700854   660530.381222 1033175.4740439   660546.413292
#Sta/Elev= 24
       0 2179.33   13.66  2171.4   27.51 2163.12    32.4 2160.32   37.94 2156.87
   41.57 2154.95   55.31 2153.89   69.08 2153.34   76.36 2153.09   98.11 2153.03
  102.08 2153.24  106.62 2156.11  110.46 2157.73  120.96 2163.32  129.34 2166.78
  137.08 2171.06  144.39 2171.28  150.58  2171.3  165.46 2171.53  173.72 2172.15
  179.43 2172.42  189.43 2173.25  199.74 2179.42  207.32 2183.21
#Mann= 3 , 0 , 0
       0      .1       0   69.08     .05       0  102.08    .065       0
Bank Sta=69.08,102.08
Exp/Cntr=0.3,0.1

Type RM Length L Ch R = 1 ,386233.9,170.92,186.6,187.89
XS GIS Cut Line= 6
 1033162.1139705  660292.5722896 1033096.6497225  660315.2843812
 1033072.6016326  660347.3484909  1033029.849446  660382.0846275
 1032976.1453667  660440.6428126 1032972.8327181  660593.8525355
#Sta/Elev= 30
       0 2177.03   10.18 2172.24   16.82 2170.51   38.08 2163.74   47.88 2161.25
   74.46 2160.12   81.86 2158.15   85.45 2157.51   86.85 2156.99   94.14 2151.28
   99.61 2148.71  113.58  2146.9  119.21 2146.48     128 2147.15  131.94  2147.9
  139.08    2150  156.46 2159.28  166.62 2165.38     170 2165.81  197.14 2166.87
     245 2166.93  259.25 2167.32  279.22 2168.44  315.55 2167.77  338.79 2169.23
  347.99  2170.3  366.36 2171.79  379.17 2193.02  385.11 2199.59   397.7 2208.81
#Mann= 3 , 0 , 0
       0      .1       0   99.61     .05       0  139.08    .065       0
Bank Sta=99.61,139.08
Exp/Cntr=0.3,0.1

Type RM Length L Ch R = 1 ,386047.3,58.6,45.19,44.09
XS GIS Cut Line= 6
  1033105.519602  660185.2328696 1032997.7376642  660190.4403844
 1032975.9857031  660197.6910179 1032905.8960844  660246.0287058
 1032860.0217256  660298.8979337 1032868.4068331  660383.2150456
#Sta/Elev= 30
       0 2178.47   18.85 2170.04   32.81 2162.93    57.3 2159.28   61.96 2159.05
   67.26  2158.3  109.35 2155.73  154.61 2154.25  166.11 2148.15  179.62 2144.96
  194.84 2144.49  207.49 2144.53  211.53 2145.63  216.53 2147.73  225.83 2150.97
  239.63 2159.55   241.1 2160.05  250.21 2160.58  253.58 2161.27  269.95 2162.14
  283.65 2160.57  286.21 2159.22  294.25 2155.91  301.49 2152.27  303.91 2151.74
  313.63 2155.96  326.97 2152.16  344.52 2159.73  368.83 2161.05  370.98 2160.87
#Mann= 3 , 0 , 0
       0      .1       0  166.11     .06       0  216.53    .065       0
#XS Ineff= 2 , 0
       0                     267       0    2162
Permanent Ineff=
       F       F
Bank Sta=166.11,216.53
Exp/Cntr=0.5,0.3

Type RM Length L Ch R = 1 ,386002.1,25.94,11.4,12.18
XS GIS Cut Line= 6
 1033080.3642187   660131.661243 1032958.2618953  660146.9364622
 1032938.9268322    660164.66027 1032851.1133754  660236.3611743
 1032825.3332611  660254.8906248 1032787.4687475  660270.1975649
#Sta/Elev= 30
       0 2170.37   22.63 2163.09   36.24 2160.06   41.11 2159.27   45.28 2159.17
   52.97 2157.86   65.27 2156.73   90.02 2154.98  112.24 2154.41   119.3 2154.33
  122.55 2154.61  133.57 2153.79  148.14 2153.33  151.24 2152.19  164.81 2149.48
  175.252145.998  187.74 2143.57  197.72 2144.79  201.06 2144.91  219.67 2144.31
  222.38 2143.95  230.62 2146.05  245.92 2151.76  252.41 2156.17  256.08  2159.5
  282.61 2161.46   291.5 2161.73   302.5 2161.73  311.04 2160.95  335.25 2176.09
#Mann= 3 , 0 , 0
       0      .1       0  175.25     .05       0  230.62     .06       0
Bank Sta=175.25,230.62
Exp/Cntr=0.5,0.3

Type RM Length L Ch R = 3 ,385996.5,,,
BEGIN DESCRIPTION:
STR_151
END DESCRIPTION:
Bridge Culvert--1,0,-1,-1, 0
Deck Dist Width WeirC Skew NumUp NumDn MinLoCord MaxHiCord MaxSubmerge Is_Ogee
0.05,11.3,2.6,0, 2, 2, , , 0.95, 0, 0,0,,
       0     300
    2155    2155
    2151    2151
       0     300
    2155    2155
    2151    2151
Pier Skew, UpSta & Num, DnSta & Num=  ,169, 2 ,215, 2 , 0 , 0 , 0 ,,
       1       1
    2140    2151
       1       1
    2140    2151
Pier Skew, UpSta & Num, DnSta & Num=  ,188, 2 ,234, 2 , 0 , 0 , 0 ,,
       1       1
    2140    2151
       1       1
    2140    2151
Pier Skew, UpSta & Num, DnSta & Num=  ,207, 2 ,253, 2 , 0 , 0 , 0 ,,
       1       1
    2140    2151
       1       1
    2140    2151
Pier Skew, UpSta & Num, DnSta & Num=  ,226, 2 ,272, 2 , 0 , 0 , 0 ,,
       1       1
    2140    2151
       1       1
    2140    2151
BR Coef=-1 , 1 , 0 ,, 0 ,,,0.8,0,2,0,
WSPro=,,,, 1 ,,,, 0 ,,,, 0 ,,,,-1 ,-1 ,-1 , 0 , 0 , 0 , 0 , 0
BR U #Sta/Elev= 69
       0 2170.37   10.09 2167.33   22.63 2163.09   25.37 2162.37    28.5 2161.72
   36.24 2160.06   41.11 2159.27   45.28 2159.17   48.57 2158.67   52.97 2157.86
   56.03 2157.55   59.41  2157.3   65.27 2156.73   72.21 2156.15   74.92 2155.94
   77.86 2155.76   79.62 2155.69   83.72 2155.37    86.7  2155.2   90.02 2154.98
   94.78 2154.82  103.34 2154.64  104.89  2154.6  110.37 2154.61  112.24 2154.41
   119.3 2154.33  122.55 2154.61  123.05 2154.59  126.61 2154.35  132.32 2153.93
  133.57 2153.79  134.32 2153.77  136.07 2153.83  148.14 2153.33  149.28 2152.84
  149.81 2152.61  151.24 2152.19  164.81 2149.84  175.252146.358  179.08 2145.08
  186.08 2143.79  187.74 2143.54  188.34 2143.59  195.62  2144.5  197.72 2144.76
  201.06 2144.88  206.03 2144.71  215.63 2144.41  219.67 2144.28  222.38 2143.92
  230.62 2146.41  245.92 2152.12  252.41 2156.17  256.08  2159.5  260.55  2159.7
  262.66 2159.92  265.47 2160.19  270.13 2160.62  276.74 2161.01  282.61 2161.46
  286.63  2161.6   291.5 2161.73  294.41 2161.79  295.21 2161.81  299.15 2161.84
   302.5 2161.73  310.95 2160.93  311.04 2160.95  335.25 2176.09
BR U #Mann= 3
       0    .065  175.25     .04  230.62     .06
BR D #Sta/Elev= 74
       0 2171.33   21.37 2164.62   29.82 2162.81   36.85  2161.4   41.54 2160.48
    45.8 2160.07   47.12 2159.92   57.25  2159.3   57.46 2159.29   58.96 2159.28
   61.57 2159.24   61.94 2159.23   62.85 2159.21   69.18 2158.92   72.63 2158.85
   75.39 2158.91   80.94 2159.19    89.7 2157.95    97.6 2156.25   99.54 2156.39
  103.74 2156.16  106.84 2156.28  110.26 2156.23  110.79 2156.26  119.11 2156.03
  119.69 2156.04  120.34 2156.01  123.65 2155.78  130.84 2155.05  132.79 2155.04
  144.24 2154.67  147.86 2154.57   154.3 2154.32  158.99 2154.12  159.53 2154.09
  164.77 2154.17  170.61 2153.95   173.5 2153.94  180.08 2154.29  180.17 2154.28
  191.07 2153.11  191.98 2152.94  196.31 2152.28  201.83 2149.86  212.76 2146.67
  216.66 2145.88   220.7 2144.53  223.19 2144.06  228.81 2143.47  239.02 2143.18
  241.74 2143.51  242.23 2143.53  250.91 2143.83   259.1 2143.55  262.24 2143.13
  265.43  2142.7  270.05 2144.09  286.32 2149.07  292.75 2151.48  299.58 2156.12
  305.16 2158.37  306.14 2159.03  307.53 2159.29  316.14 2160.39  317.25 2160.51
  318.31 2160.59  324.54 2160.95  330.86  2161.2  332.03 2161.27  339.61 2161.49
  344.63  2161.7  345.74  2161.6  353.87 2161.12  375.32 2174.51
BR D #Mann= 3
       0    .065   220.7     .04  250.91     .06
BC Design=,, 0 ,, 0 ,,,,,,

Type RM Length L Ch R = 1 ,385990.7,91.17,96.22,95.41
XS GIS Cut Line= 6
 1033086.8859691  660066.4435882 1032977.8793283  660085.5430454
 1032955.8449973  660128.4070117 1032935.7043217  660153.3814832
 1032836.6120479  660233.1386638  1032784.246237  660255.6962373
#Sta/Elev= 30
       0 2171.33   21.37 2164.62   41.54 2160.48   57.46 2159.29   72.63 2158.85
   80.94 2159.19    89.7 2157.95    97.6 2156.25  119.69 2156.04  130.84 2155.05
  159.53 2154.09   173.5 2153.94  180.08 2154.29  196.31 2152.28  201.83 2149.86
   220.7 2144.53  228.81 2143.47  239.02 2143.18  250.91 2143.83   259.1 2143.55
  265.43  2142.7  286.32 2149.07  292.75 2151.48  299.58 2156.12  306.14 2159.03
  317.25 2160.51  324.54 2160.95  344.63  2161.7  353.87 2161.12  375.32 2174.51
#Mann= 3 , 0 , 0
       0    .065       0   220.7     .05       0  250.91     .06       0
Bank Sta=220.7,250.91
Exp/Cntr=0.5,0.3

Type RM Length L Ch R = 1 ,385894.5,341.06,338.14,351.37
XS GIS Cut Line= 6
 1032954.9157401  659931.0366423 1032949.1973927  660020.9986715
  1032906.434703   660071.949969 1032871.8606213  660094.6960818
 1032818.1797878  660113.8028032 1032738.1134804   660206.606935
#Sta/Elev= 30
       0 2169.92   29.21 2167.43   31.95 2166.32   60.66 2156.81   67.16 2153.79
   90.78    2153  111.74 2151.68  122.85  2151.4  135.15 2150.22  140.39 2150.31
  161.88 2147.61  172.98 2146.94  180.67 2147.12  186.48 2146.17  200.71 2145.47
  209.56 2142.12  217.64  2141.7  222.52 2141.67  230.45 2140.75  237.88 2141.37
  251.01  2143.9  300.77 2153.92   303.5 2154.92  315.89 2158.54  342.72 2160.54
  355.18 2160.58  356.82 2161.59  374.95  2184.9  376.48 2188.94  378.45 2190.31
#Mann= 3 , 0 , 0
       0     .08       0  217.64     .05       0  251.01     .07       0
Bank Sta=217.64,251.01
Exp/Cntr=0.3,0.1

Type RM Length L Ch R = 1 ,385556.4,421.69,401.98,403.53
XS GIS Cut Line= 4
 1032807.8980282  659762.2395465  1032735.086501  659784.9931658
 1032518.9273753  659905.5872056 1032437.0144186  660014.8044509
#Sta/Elev= 30
       0 2197.4469.43997 2157.2381.87997 2150.9392.28998 2144.71  103.86 2138.77
  109.83 2136.34  114.98 2135.88  126.07 2135.67  131.75 2136.74  136.22 2137.58
  151.52 2141.44  169.61 2144.22   179.1 2145.25  261.75 2147.05  307.27 2149.18
  318.71 2150.06  324.88  2150.9  329.75 2152.58  335.87 2155.36  341.04 2156.81
  348.92 2158.35  360.69 2158.07  383.26 2156.54  396.12 2157.02  422.74 2160.42
  428.11 2161.36  437.15  2163.8  443.05  2164.9  448.23 2165.38  460.33  2167.4
#Mann= 4 ,-1 , 0
       0      .1       0  103.86     .05       0  131.75     .08       0
  151.52     .05       0
Bank Sta=103.86,131.75
Exp/Cntr=0.3,0.1

Type RM Length L Ch R = 1 ,385154.4,803.48,700.13,320.7
XS GIS Cut Line= 6
 1032564.4345533  659432.3124456 1032464.3187375  659480.0949885
 1032343.7246977  659584.7615342 1032289.1160599  659680.3266201
 1032245.8842166   659750.862752 1032204.9277685  659800.9206599
#Sta/Elev= 30
       0  2154.9    9.35 2152.35   22.17 2149.93   60.55 2134.25   81.04 2129.83
   94.01 2131.25  107.57 2135.77  129.06 2139.46  146.51 2139.83  196.45 2139.21
  211.57 2140.11  246.38 2141.18  256.69 2141.97  266.89    2143  288.49 2146.72
   321.7 2152.98  365.85 2159.23  374.27 2160.83  386.57 2160.94  402.97 2158.53
  433.83 2156.59  448.31 2156.24  458.18 2157.65  461.75 2158.56  476.98 2173.54
  483.92 2177.12  489.64 2181.01  507.96 2191.25  520.98 2194.08  528.09 2196.48
#Mann= 4 ,-1 , 0
       0      .1       0   60.55     .05       0  107.57     .08       0
  129.06     .05       0
#XS Ineff= 2 , 0
       0                   142.3       0    2142
Permanent Ineff=
       F       F
Bank Sta=60.55,107.57
Exp/Cntr=0.3,0.1

Type RM Length L Ch R = 1 ,384454.3,75.98,73.15,57.45
XS GIS Cut Line= 6
 1031881.2602973  659129.2804708 1031892.6567054  659161.3975797
 1032030.4494642  659289.8660155 1032035.6590069  659407.4490272
 1032065.3564634  659528.9385451  1032045.558149  659671.1263051
#Sta/Elev= 30
       0 2175.85   23.74 2163.81   28.32 2160.96   34.08 2155.81   49.52 2144.61
   73.22 2128.07   79.72 2123.74   88.73 2124.02  107.68 2126.77  117.21 2128.02
  122.49 2129.13  144.86 2130.84  172.91 2132.08  236.67 2132.85  252.18 2133.76
  259.44 2134.85  266.54 2134.54   288.6 2134.73   344.8 2134.25  422.75 2135.98
  459.75 2137.78  480.77 2139.72  517.36 2144.27   541.5  2149.7  550.92 2152.51
  560.17 2154.58  573.75 2155.46  587.02 2154.85  600.45 2153.44  612.02 2159.58
#Mann= 3 , 0 , 0
       0      .1       0   73.22     .05       0  107.68     .05       0
Bank Sta=73.22,107.68
Exp/Cntr=0.5,0.3

Type RM Length L Ch R = 1 ,384381.1,22.99,20.85,85.36
XS GIS Cut Line= 6
 1031827.3864449  659151.0372142 1031837.7468104   659199.730914
  1031980.719752  659316.8029417 1031983.4635139  659405.6491722
   1032020.36033   659615.331102 1032010.4611879  659663.0269877
#Sta/Elev= 30
       0 2175.86     8.6 2171.49   39.11 2143.55   59.58  2138.4   72.74 2130.52
   90.53 2124.31  104.17 2122.93  107.04  2123.6  116.43 2123.69  136.91  2123.2
  151.29 2124.74  153.73 2125.59  161.53  2127.2   180.6 2138.22   202.4 2136.69
  206.88 2135.71   215.6 2136.12   224.4 2135.19  251.86 2134.38  323.34 2133.42
   401.3 2135.03  440.66 2136.62  465.02 2140.47  487.79 2142.04  504.13 2144.15
  515.03 2146.69  533.88 2153.66  546.49 2155.49  575.21 2153.75   585.3 2158.76
#Mann= 3 , 0 , 0
       0      .1       0   90.53     .05       0  153.73     .05       0
Bank Sta=90.53,153.73
Exp/Cntr=0.5,0.3

Type RM Length L Ch R = 3 ,384371. ,,,
BEGIN DESCRIPTION:
STR_150
END DESCRIPTION:
Bridge Culvert--1,0,-1,-1, 0
Deck Dist Width WeirC Skew NumUp NumDn MinLoCord MaxHiCord MaxSubmerge Is_Ogee
2,18,2.6,0, 2, 2, , , 0.95, 0, 0,0,,
       0     190
    2136    2136
  2133.5  2133.5
       0     198
    2136    2136
  2133.5  2133.5
Pier Skew, UpSta & Num, DnSta & Num=  ,119, 2 ,128, 2 , 0 , 0 , 0 ,,
       3       3
    2120  2133.5
       3       3
    2120  2133.5
BR Coef=-1 , 1 , 0 ,, 0 ,,,0.8,0,2,0,
WSPro=,,,, 1 ,,,, 0 ,,,, 0 ,,,,-1 ,-1 ,-1 , 0 , 0 , 0 , 0 , 0
BC Design=,, 0 ,, 0 ,,,,,,

Type RM Length L Ch R = 1 ,384360.3,60.11,104.36,60.13
XS GIS Cut Line= 6
 1031813.9179818  659151.0372142 1031825.3143597  659215.2714321
 1031928.9179545  659303.3344786 1031931.2679906   659412.848562
 1031899.7707093  659600.0324251 1031906.0701716   659661.227163
#Sta/Elev= 30
       0  2172.4    7.52    2169    35.8 2151.13   47.24 2140.71      53 2139.06
   57.98  2139.7   87.22 2128.36   98.25 2124.22  116.56  2122.8  126.02 2125.07
  147.78 2124.18  161.63 2125.79  167.28 2127.11  176.89 2128.11   180.8 2130.49
  193.83 2135.76  201.41 2135.89  215.52 2133.76  232.34 2132.61  312.53 2132.47
  400.52 2135.19  410.09 2136.28  418.82 2136.24   466.8 2139.03  472.06 2139.54
  485.51 2145.72  497.71 2153.44   508.4 2154.82  543.04 2153.49  562.29 2147.66
#Mann= 3 , 0 , 0
       0      .1       0   87.22     .05       0  161.63     .05       0
Bank Sta=87.22,161.63
Exp/Cntr=0.5,0.3

Type RM Length L Ch R = 1 ,384255.9,217.77,259.92,316.43
XS GIS Cut Line= 6
 1031776.6764437  659156.9677401  1031778.012442  659295.9122862
 1031818.0926018  659374.7366077 1031835.4606701   659493.641089
 1031873.6729628    659534.33808 1031860.1741409  659657.6274529
#Sta/Elev= 30
       0 2168.56    6.17 2163.29   47.15 2138.64   50.81 2137.63   59.25  2137.3
   70.84 2130.47   82.42 2129.25   95.46 2125.68  107.73 2122.32  110.52 2123.06
  118.94 2122.96   130.6 2126.71  193.03 2124.72  224.84 2130.53  231.34 2131.11
  332.25 2133.15  388.85 2136.19  411.63  2139.5  426.25 2138.34  439.72 2142.91
  452.45 2147.87   457.7 2150.54  473.71 2154.13  476.75 2154.33  493.53 2153.88
  504.29 2152.72  512.25 2149.27  522.56 2146.36   530.2 2145.36  531.53 2145.72
#Mann= 3 , 0 , 0
       0      .1       0   95.46     .05       0   130.6    .055       0
Bank Sta=95.46,130.6
Exp/Cntr=0.3,0.1

Type RM Length L Ch R = 1 ,383996.0,195.42,206.94,209.53
XS GIS Cut Line= 6
 1031654.3326726  659167.3191161 1031568.6467217  659283.7641728
 1031551.0701071  659351.8735394 1031555.4642607  659435.3624286
 1031676.3034409  659545.2162398 1031660.9239182  659644.0846819
#Sta/Elev= 30
       0 2133.42    3.48 2131.56   10.84  2130.3   29.82 2129.32   63.88 2128.48
   89.59    2127  102.57 2126.77     113 2127.49  133.31 2126.45  161.64 2126.26
   192.4 2122.28  210.44    2119  221.31 2117.86  230.84 2117.75  236.35 2117.92
  241.95 2119.09  280.68 2127.43  313.36 2131.03  355.76 2134.34   364.3 2137.53
  378.98 2147.52  414.17 2148.76  427.37 2151.36  448.48  2153.3   454.5 2154.53
  504.77  2152.6  519.42 2153.56  533.67 2156.78  545.61 2161.69  561.89 2167.05
#Mann= 3 , 0 , 0
       0      .1       0  210.44     .05       0  241.95     .06       0
Bank Sta=210.44,241.95
Exp/Cntr=0.3,0.1

Type RM Length L Ch R = 1 ,383789.0,179,286.51,351.24
XS GIS Cut Line= 6
 1031478.7472564  659062.1113487 1031350.4907267  659263.8481765
 1031341.1387086  659331.9844513 1031354.4987518  659406.8007477
 1031346.4827319  659448.2169058 1031319.7626152   659477.609019
#Sta/Elev= 30
       0 2130.38  120.94 2125.75  134.06 2125.61   147.8 2126.18  158.54 2125.15
  169.97 2124.83     185 2123.42   194.5 2123.51  207.03 2122.89  209.84 2123.32
  234.38 2123.69  255.65  2122.4  270.29 2120.05  273.76    2120  295.11 2124.48
  300.34 2124.58   322.5  2119.3  331.94 2115.86  336.21 2115.43  342.84 2116.04
  357.09 2116.22  366.88 2119.12  372.44    2121  380.37 2124.38  407.29 2128.75
  434.45 2129.21  441.11 2129.76  453.23 2133.12  465.53 2142.32  467.28 2143.16
#Mann= 3 , 0 , 0
       0      .1       0   322.5     .05       0  366.88     .07       0
#XS Ineff= 2 , 0
       0  300.34 2124.58               0
Permanent Ineff=
       F       F
Bank Sta=322.5,366.88
Exp/Cntr=0.3,0.1

Type RM Length L Ch R = 1 ,383502.5,470.06,400.58,392.39
XS GIS Cut Line= 6
 1031397.2747593  658949.8085857 1031321.0986135  658996.6471007
 1031254.2983673  659150.2877185 1031235.5942705  659170.3277833
  1031140.783281  659190.8862175 1031044.5455196  659235.7920616
#Sta/Elev= 30
       0 2139.24    33.7 2136.58   83.49  2133.8  125.11 2132.75  134.93 2131.85
  164.78 2130.46  188.72 2131.23  192.69 2131.13  215.76 2128.99  231.54 2128.38
  239.02  2126.8  257.58 2124.15  274.14 2122.68  335.47 2118.73  345.03 2118.48
  346.82 2118.24  355.66 2115.44  361.57 2112.96  362.71 2112.87  379.39 2113.35
  382.65 2113.91  390.65 2117.25  420.79 2130.72  430.21 2133.22   439.3  2137.4
     444 2139.05  464.97 2145.05  471.66  2146.2  478.86 2148.89  489.64 2148.86
#Mann= 3 , 0 , 0
       0    .065       0  355.66     .05       0  390.65     .08       0
Bank Sta=355.66,390.65
Exp/Cntr=0.3,0.1

Type RM Length L Ch R = 1 ,383101.9,190.01,378.53,452.99
XS GIS Cut Line= 4
 1031405.1845083  658623.5688206 1031049.9062508  658766.1327207
   1030963.91535  658831.7573587 1030839.4547879  658931.3257781
#Sta/Elev= 30
       0 2137.4910.79999 2136.32   27.38 2133.6559.02002  2125.883.14001 2124.24
  105.06 2123.93  117.85 2122.09  128.07  2121.4  150.82 2117.89  169.98 2118.74
  191.99 2117.82  228.45 2117.71   244.1  2117.3  250.89 2117.88   292.7 2117.88
  304.41  2118.4  417.81 2118.81  475.16 2118.01  496.86 2117.36  498.76 2117.33
     516 2112.41  526.49 2109.24  542.43 2112.08  554.48 2113.98  562.44 2115.25
  579.14 2116.31  602.27 2119.47  612.37 2122.07   629.7 2123.99  650.37  2129.5
#Mann= 5 ,-1 , 0
       0     .05       0  496.86     .08       0     516     .05       0
  542.43     .08       0  554.48     .06       0
#XS Ineff= 2 , 0
       0  417.81 2118.81               0
Permanent Ineff=
       F       F
Bank Sta=516,542.43
Exp/Cntr=0.3,0.1

Type RM Length L Ch R = 1 ,382723.4,200.88,395.44,407.51
XS GIS Cut Line= 5
 1030733.0976244  658485.5307702 1030968.4411694  658585.0992198
 1031185.6813765  658499.1082888 1031237.7285261  658490.0566198
 1031298.8273447  658453.8499136
#Sta/Elev= 30
       0 2144.67   33.61 2127.24   42.64 2115.31   49.02 2111.37   71.97 2109.25
   73.93 2108.59   78.75 2106.96   90.19 2106.79   94.04 2107.57   100.6 2108.61
  115.43 2112.42  194.59 2116.52  211.11    2117   249.1 2117.28  306.67 2116.93
  318.74 2117.45   329.8 2116.58  363.15 2116.48  387.46 2115.34  415.67 2114.76
  448.65 2115.54  457.48 2115.26  491.89 2115.16  496.11 2116.23  524.16 2119.31
  527.65 2120.07  548.79 2122.14  552.32 2122.21  563.16 2120.82  613.03  2139.1
#Mann= 3 , 0 , 0
       0     .05       0   73.93     .05       0   94.04     .08       0
Bank Sta=73.93,94.04
Exp/Cntr=0.3,0.1

Type RM Length L Ch R = 1 ,382328.0,187.82,187.71,159.8
XS GIS Cut Line= 5
 1031321.6784874  658316.3830804 1031287.9689499  658301.0605826
 1031186.8403676  658291.8670779 1030979.9864355  658158.5612139
 1030917.1641582  658143.2386858
#Sta/Elev= 30
       0 2140.46    26.4 2125.72   33.37 2122.63   42.79 2117.18   60.64 2117.44
   74.18 2117.27   78.52 2116.16   82.77 2116.05   91.27 2114.43  109.21 2114.07
  110.84 2114.25  130.53 2113.16  148.02 2112.69  197.71 2112.78  235.46 2110.92
  256.61 2109.62  274.97 2108.96  286.82 2108.91   296.6 2108.05  320.05 2103.38
   325.1 2102.31  332.32 2102.59  340.18 2103.48  347.23  2104.4  358.54 2107.74
   389.8  2110.8  403.46 2111.54  413.46 2115.81   431.4 2120.38  449.33 2128.71
#Mann= 3 , 0 , 0
       0     .05       0  320.05     .05       0  340.18     .08       0
Bank Sta=320.05,340.18
Exp/Cntr=0.3,0.1

Type RM Length L Ch R = 1 ,382140.3,691.59,496.9,128.13
XS GIS Cut Line= 4
 1031371.2407269  658184.5625569   1031344.08572  658130.2525127
 1031052.1691756  658005.7919808 1030945.8119818  657999.0032064
#Sta/Elev= 30
       0 2128.4814.73001 2122.7628.39001 2118.4847.12003 2115.8961.95001 2114.47
87.95001 2114.23  163.21 2108.82  184.99 2107.92   215.9 2107.24  239.28 2107.66
  245.87  2106.9  257.56  2106.7  262.24  2105.1  270.16 2101.52  277.82 2100.87
  292.04 2105.08  293.38 2105.55  300.58 2105.48  319.47 2106.52  332.36 2106.18
  358.52 2106.55  360.75    2106  381.29  2104.1   401.9 2107.59  427.24 2110.02
  438.89 2112.44  448.07 2114.92  468.33 2125.95  476.32 2129.89  484.64 2136.01
#Mann= 4 ,-1 , 0
       0     .05       0  245.87     .08       0  262.24     .05       0
  292.04      .1       0
#XS Ineff= 2 , 0
       0                  326.09       0 2106.63
Permanent Ineff=
       F       F
Bank Sta=262.24,292.04
Exp/Cntr=0.3,0.1

Type RM Length L Ch R = 1 ,381643.4,212.43,246.08,240.05
XS GIS Cut Line= 6
 1031043.2095213  657758.1701399 1031029.8494478  657808.9383464
 1031004.4653597   657851.690533 1030979.0812413  657887.7626678
 1030955.0331515   657917.154781 1030917.6250184  657954.5629443
#Sta/Elev= 28
       0 2137.98   30.28 2121.62    52.5 2110.61    69.2 2102.86   71.63 2101.58
   81.83 2098.08   82.37  2097.9   84.65 2097.12   84.79 2097.09   86.02 2097.11
   97.51 2097.42   102.1 2098.24  102.22 2098.29  103.68 2098.85  120.39 2105.38
  146.33 2115.21  152.13 2117.61  175.04  2125.8  176.99 2126.39  179.54 2127.86
   180.4 2128.21  184.31 2129.97  209.83  2141.2  209.93 2141.24  210.58 2141.47
   216.7 2141.53  231.07 2147.85  237.25 2150.49
#Mann= 3 , 0 , 0
       0      .1       0   81.83     .05       0  103.68      .1       0
Bank Sta=81.83,103.68
Exp/Cntr=0.3,0.1

Type RM Length L Ch R = 1 ,381397.3,189.55,224.31,266.64
XS GIS Cut Line= 6
 1030859.8086106  657740.8961445 1030808.7669632  657787.0766941
 1030785.6766732  657796.7989199  1030772.308609   657807.736405
 1030743.1419619  657852.7016954  1030735.850285  657874.5766958
#Sta/Elev= 20
       0 2140.29     4.4 2137.97   42.97 2112.74    53.4 2105.96   57.45 2103.34
   60.49 2101.94   68.97 2101.09   80.67 2099.67   81.66 2099.55   94.17  2098.2
   95.59  2098.3  100.76 2099.35  111.45  2102.1  115.17 2103.03  132.98 2109.09
   151.4 2114.32  165.11  2118.5  170.01 2119.98  182.85 2126.56  188.17 2129.88
#Mann= 3 , 0 , 0
       0      .1       0   68.97     .05       0  111.45      .1       0
Bank Sta=68.97,111.45
Exp/Cntr=0.3,0.1

Type RM Length L Ch R = 1 ,381173.0,191.65,303.61,254.42
XS GIS Cut Line= 6
 1030774.7391881  657620.5836271 1030713.9752846  657632.7364017
 1030654.4266707  657638.8127891 1030630.1211215  657635.1669809
 1030605.8155722  657636.3822402 1030575.4336053  657657.0419813
#Sta/Elev= 28
       0 2129.27    18.5 2121.18   43.83 2112.93   67.75 2105.44   77.15 2104.77
   82.59  2103.9   88.63 2103.17   90.53 2102.29    91.8 2101.78   94.35 2100.32
   97.52 2098.79  101.65 2097.62  104.19 2096.68  110.21 2096.24  115.95 2098.57
  118.49 2100.61  121.66  2102.8  128.65 2104.41  146.63 2109.26  147.71 2109.43
  161.02 2109.93  163.64 2110.48  171.03 2111.83  181.19 2112.82   182.5 2113.37
  200.37 2120.72  205.98 2123.19  207.79 2124.37
#Mann= 3 , 0 , 0
       0      .1       0   88.63     .04       0  121.66      .1       0
Bank Sta=88.63,121.66
Exp/Cntr=0.3,0.1

Type RM Length L Ch R = 1 ,380869.4,79.73,316.98,373.71
XS GIS Cut Line= 6
 1030717.6211231  657517.2850124 1030700.6072204  657507.5628169
  1030667.794735   657466.243365 1030594.8780569  657433.4308492
 1030487.9336037  657409.1252999 1030410.1558278  657494.1947527
#Sta/Elev= 30
       0 2111.02    9.58 2108.84   20.73 2105.56   22.52 2105.31   41.26 2104.35
   55.04 2103.26   76.15 2102.88   88.04 2102.92  101.72 2102.73  117.06 2102.33
  151.01 2101.89  155.74 2101.64  171.66 2100.37  174.74  2100.4  186.28 2099.51
  212.23 2100.09  225.38 2101.07  227.82 2101.09  241.74 2100.42  252.33 2100.13
  261.74 2099.25  264.74 2099.21  281.68 2096.29  292.83 2094.46  295.33 2094.27
  301.71 2096.24   346.2 2109.94  347.19 2110.45  364.51 2122.48   377.8 2131.42
#Mann= 3 , 0 , 0
       0      .1       0  281.68     .05       0  301.71      .1       0
Bank Sta=281.68,301.71
Exp/Cntr=0.3,0.1

Type RM Length L Ch R = 1 ,380552.4,368.98,333.43,286.51
XS GIS Cut Line= 6
 1030738.2808339  657483.2572373 1030711.5447358  657410.3405895
 1030673.8711223  657379.9586226 1030661.7183476  657358.0836222
 1030621.6141853  657247.4933609 1030579.0794438  657215.8961347
#Sta/Elev= 30
       0 2109.02    3.99 2108.14   32.21 2104.22   42.97 2102.31   58.67 2101.23
   79.03  2100.8  108.91  2101.3   120.9 2100.45  126.11 2099.53  162.52 2094.09
  183.09 2090.98  189.34 2092.55  197.79 2093.39  203.03 2094.21  211.02 2093.21
  213.61 2093.21  218.34 2092.34  220.16  2092.6  231.22 2096.22  244.61 2097.67
  256.12 2098.35  260.29 2098.83  266.66 2099.13  269.27 2100.09  287.66 2107.97
  298.28 2112.95  301.08 2113.87  316.04 2119.64  318.36 2120.35  322.82 2122.59
#Mann= 3 , 0 , 0
       0     .07       0  162.52     .05       0  197.79      .1       0
Bank Sta=162.52,197.79
Exp/Cntr=0.3,0.1

Type RM Length L Ch R = 1 ,380219. ,421.28,466.51,472.78
XS GIS Cut Line= 5
 1031096.4551921  657354.2304481 1031083.7262967  657263.5369025
 1030872.1080033  657117.1543641 1030849.8324062  657055.1008631
 1030646.1697178  656994.6385195
#Sta/Elev= 30
       0 2122.27   10.12 2117.53    23.5 2112.54    35.9 2106.76   42.35 2105.49
   57.98 2100.34   65.39 2099.37   95.96 2097.48  178.83 2097.39  224.63 2096.05
  244.752091.972  253.96 2089.14     272 2088.58  284.49 2088.91  309.43 2091.96
     342  2093.4  370.24 2096.02  372.31 2095.72  378.23 2098.41  385.27 2099.84
  391.84 2099.18  400.37 2099.67  418.92 2098.36  455.03 2097.46  491.69 2097.98
  525.19 2097.22  575.01 2098.05  597.39 2100.02  603.44  2102.1  627.27 2119.71
#Mann= 3 , 0 , 0
       0    .055       0  244.75     .05       0  309.43     .08       0
Bank Sta=244.75,309.43
Exp/Cntr=0.3,0.1

Type RM Length L Ch R = 1 ,379752.4,64.2,163.4,200.2
XS GIS Cut Line= 5
 1031475.1405242  657039.1897137 1031336.7135302  656980.3184669
 1031238.0644099  656803.7047264 1031117.1396924  656725.7401063
 1030725.7254649  656719.3756587
#Sta/Elev= 30
       0 2111.6625.91998 2102.3541.14001 2098.5372.29999  2094.9  117.14 2092.44
  123.61 2093.56   146.4 2092.55  177.72 2093.34  247.62  2092.6  253.34 2091.96
  258.86 2088.34  261.17 2086.12  283.07 2085.92  287.39 2086.83  291.35 2088.63
   305.6 2093.45  313.96 2093.58  319.82 2092.19  344.43 2089.76  366.38  2089.3
  401.36 2091.63  487.14  2095.6   515.4 2096.16  586.86 2092.98  696.36 2093.15
  797.23 2092.15  835.28 2092.81  854.45 2096.36  874.62  2109.3  888.07 2119.74
#Mann= 3 ,-1 , 0
       0    .055       0  258.86     .05       0  291.35    .055       0
#XS Ineff= 2 , 0
       0  123.61    2100     370       0    2100
Permanent Ineff=
       F       F
#Block Obstruct= 1 ,-1
  452.23  545.22 2107.08
Bank Sta=258.86,291.35
Exp/Cntr=0.5,0.3

Type RM Length L Ch R = 1 ,379589.0,166.73,130.2,133.92
XS GIS Cut Line= 6
 1031615.0284626  656872.0214286 1031536.2845027  656827.5139717
 1031455.2580648  656812.6781527 1031311.4647097  656739.6402513
 1031156.2591769  656708.8273895 1030730.2172046  656678.0486837
#Sta/Elev= 30
       0 2129.67    16.5 2109.89    18.2 2106.99   31.16 2103.92   78.63 2100.66
   90.71 2100.79  114.29 2096.53  160.64 2098.03   183.6 2097.31  197.62 2092.07
  212.53 2089.32  216.93 2086.99  218.61 2086.11   239.5 2085.61  246.01 2087.09
  263.94 2090.47  297.77 2090.95  318.99 2093.77  325.96 2095.91  340.16 2097.22
  403.53 2096.28  428.23 2094.38   439.6 2092.37  498.99 2095.17  555.89 2095.59
   614.7 2092.85  653.84 2092.37  839.77    2092     891    2094     922    2116
#Mann= 3 , 0 , 0
       0    .055       0  216.93    .045       0  246.01    .055       0
#XS Ineff= 3 ,-1
       0   178.5    2097   320.5  347.67    2097  347.67     922    2100
Permanent Ineff=
       F       F       F
#Block Obstruct= 1 ,-1
     460     550    2100
Bank Sta=216.93,246.01
Exp/Cntr=0.5,0.3

Type RM Length L Ch R = 3 ,379532. ,,,
BEGIN DESCRIPTION:
STR_146
END DESCRIPTION:
Bridge Culvert--1,0,-1,-1, 0
Deck Dist Width WeirC Skew NumUp NumDn MinLoCord MaxHiCord MaxSubmerge Is_Ogee
50,12,2.6,0, 6, 8, , , 0.95, 0, 0,0,,
       0   188.5   188.5   290.5   290.5  340.16
    2097    2097    2097    2097    2097    2097
                    2095    2095
     100  207.87  207.87  309.87  309.87     407     527     550
    2097    2097    2097    2097    2097    2096    2094    2093
                    2095    2095
BR Coef=-1 , 1 , 0 ,, 0 ,,,0.8,-1,2,0,
WSPro=,,,, 1 ,,,, 0 ,,,, 0 ,,,,-1 ,-1 ,-1 , 0 , 0 , 0 , 0 , 0
BC Design=,, 0 ,, 0 ,,,,,,

Type RM Length L Ch R = 1 ,379458.8,150.31,140.82,71.36
XS GIS Cut Line= 6
 1031685.7839466  656624.3773104 1031528.2959661  656663.1787087
 1031419.8803379  656650.6253072 1031250.9802099  656596.9880898
 1031094.6334533   656591.282001  1030704.235397  656637.8296105
#Sta/Elev= 30
       0  2112.1   11.55 2105.14   48.81 2104.39   97.23 2101.62  107.77 2101.42
  134.75 2092.79  152.27 2092.47  200.84 2090.48  208.96  2090.8   217.2 2091.67
  233.51 2090.12  242.82 2086.64  250.44 2085.36   259.3 2084.73  267.87 2084.82
  283.16 2086.65   297.1 2087.99  338.01 2089.67  401.29 2089.51  451.02 2091.51
  505.26 2091.69  545.73 2093.49  587.88 2093.42  613.98 2092.68  722.09 2091.07
  783.49 2090.83  837.97 2091.13  868.85 2090.73     968    2094    1001    2116
#Mann= 3 , 0 , 0
       0    .055       0  242.82    .045       0  283.16    .055       0
#XS Ineff= 3 ,-1
       0  187.65    2094  330.17  559.97    2094  559.97    1001    2095
Permanent Ineff=
       F       F       F
Bank Sta=242.82,283.16
Exp/Cntr=0.5,0.3

Type RM Length L Ch R = 1 ,379318.0,808.34,609.12,390.26
XS GIS Cut Line= 6
 1031563.9654157  656468.2038379 1031511.5238743  656511.4680982
 1031261.1155936  656506.2239592 1031230.9616959   656561.287555
 1031013.3293672  656545.5550774 1030709.1684876  656647.8160756
#Sta/Elev= 30
       0 2148.84    6.15 2148.89    8.87 2147.49   61.21 2093.43    74.3 2090.51
   79.14 2090.79   91.71 2089.71   99.83 2090.01  108.84 2086.89  133.69 2085.55
  159.72 2084.12  170.21 2084.88  178.26 2086.97   189.3 2088.65  200.75 2088.73
  218.26 2087.75  246.57 2088.14  273.91 2091.12  312.63 2090.14   393.1 2090.99
  452.27 2093.16  566.69 2092.83  611.29 2091.46  675.72  2090.4  771.31    2090
  873.69 2092.84  883.63 2093.25  896.39  2096.9  914.86 2112.12     921 2116.35
#Mann= 3 , 0 , 0
       0      .1       0  133.69     .05       0  178.26    .055       0
#XS Ineff= 2 , 0
       0                  494.44       0    2100
Permanent Ineff=
       F       F
#Block Obstruct= 1 ,-1
  304.46  408.92  2111.7
Bank Sta=133.69,178.26
Exp/Cntr=0.3,0.1

Type RM Length L Ch R = 1 ,378708.8,395.71,343.33,318.9
XS GIS Cut Line= 6
 1030796.6009311  655954.8171367 1030819.0063476  656015.6319206
 1030918.2304385  656153.2653185 1030899.0257699  656463.7406733
 1030726.1838129  656527.7562051 1030678.1721716   656556.563208
#Sta/Elev= 30
       0 2119.25   36.21 2100.74   49.97 2094.51    54.3 2093.84   99.92 2090.64
  175.49 2090.32  195.79 2089.43  207.64 2088.03  283.49 2087.44  310.48 2088.45
  331.58 2086.43  359.72 2085.14  367.15 2084.41  371.07 2083.34  384.48 2080.04
  395.03 2079.23  412.72 2079.07  431.61  2084.5  449.71 2087.88  467.71 2089.49
  488.66 2089.68  510.65 2091.18  638.57 2089.17  712.21 2090.75  734.06 2091.76
  741.34 2094.34  753.24 2109.87  767.23 2124.85  771.46 2127.85  785.86 2134.87
#Mann= 3 , 0 , 0
       0      .1       0  371.07     .05       0  431.61     .06       0
Bank Sta=371.07,431.61
Exp/Cntr=0.3,0.1

Type RM Length L Ch R = 1 ,378365.5,501.97,459.67,418.95
XS GIS Cut Line= 6
 1030503.7322168  656167.1114049 1030554.7738945  656258.2572449
 1030573.0030564  656339.6808592 1030599.7391849  656387.0766985
 1030599.7391849  656417.4586351 1030591.2322184   656435.687797
#Sta/Elev= 30
       0 2133.25   12.85 2123.11   21.22 2114.29   32.07 2105.85   40.15 2100.31
   58.12 2094.01   83.32 2088.71   90.41 2086.81  103.39 2085.05  148.86  2077.9
  154.62    2077  173.82 2076.95  185.58  2077.7  187.07 2078.27  189.53  2079.2
  195.09 2080.85  199.66 2085.37  202.61 2087.84  208.59 2089.08   213.4 2089.81
  217.87 2091.23  218.96 2091.22  225.62 2091.94  232.39 2092.14  252.78 2091.46
  268.38 2091.59  274.59 2093.02   275.2 2093.26  286.18 2103.02  294.71  2112.6
#Mann= 3 , 0 , 0
       0      .1       0  148.86     .05       0  187.07    .055       0
Bank Sta=148.86,187.07
Exp/Cntr=0.3,0.1

Type RM Length L Ch R = 1 ,377905.9,296.77,301.43,298.37
XS GIS Cut Line= 6
  1030152.516951   656534.125314  1030175.607241  656558.4308633
 1030215.7114033   656568.153089 1030276.4752765  656607.0419618
 1030291.0586303  656619.1947365 1030316.5794389  656632.5628007
#Sta/Elev= 22
       0 2117.27   12.52 2105.59   33.52 2083.13   37.31 2079.55   42.28 2075.68
   44.54 2074.91   57.95 2073.54   65.27 2073.43   73.49 2073.58   91.76 2076.24
  101.99 2077.77   109.9 2079.82  131.71 2085.16  136.09 2087.93  141.45  2091.2
  150.27 2095.77   164.4 2095.94  172.04 2096.46  178.14 2096.03   178.6 2096.06
  186.28 2098.04  194.92 2105.67
#Mann= 3 , 0 , 0
       0      .1       0   37.31     .05       0   91.76     .08       0
Bank Sta=37.31,91.76
Exp/Cntr=0.3,0.1

Type RM Length L Ch R = 1 ,377604.4,174.4,188.28,198.09
XS GIS Cut Line= 6
 1030080.8155625  656785.6878035 1030102.6905629  656812.4239017
 1030107.5516606  656839.1600301 1030135.5030483  656853.7433536
 1030216.9266626  656903.5697417 1030219.3572418   656916.937806
#Sta/Elev= 29
       0 2119.63     .55 2119.15   34.54 2098.12   34.84 2097.97   35.31 2097.86
   61.72  2087.4   62.05 2087.22   66.24 2083.38   78.89 2078.06   86.19 2074.58
   92.38 2072.26   93.25 2071.93   95.78 2071.02   99.24    2071  106.37 2070.86
  111.83 2070.83  112.49 2070.81  113.61 2070.78  119.45    2074  145.72  2087.4
  149.62 2089.66  177.99 2106.06  183.82 2109.27  185.23 2109.33  188.74 2109.76
  192.79 2110.29  192.96 2110.32  199.09 2110.84  202.33 2111.21
#Mann= 3 , 0 , 0
       0      .1       0   86.19     .05       0  119.45     .08       0
Bank Sta=86.19,119.45
Exp/Cntr=0.3,0.1

Type RM Length L Ch R = 1 ,377416.1,82.99,122.53,142.91
XS GIS Cut Line= 6
  1029967.794722  656924.2294828 1030010.3294635  656989.8544841
 1030057.7252725  657038.4655826 1030066.2322389  657059.1252935
 1030068.6627878   657083.430873 1030063.8016598  657104.0905838
#Sta/Elev= 27
       0 2106.22   25.14 2092.36   31.54 2089.32   41.42 2085.08    45.3 2082.79
   49.87 2075.26   51.56 2072.73   52.75 2072.23   56.96 2071.27   93.57 2070.03
  102.28 2070.43  104.34 2070.92  109.34 2073.31  115.51 2075.83  117.57 2076.51
  127.91 2081.73  132.12 2084.04   138.5  2085.8  142.51 2087.54  147.02 2089.87
  151.28 2092.66  168.68 2097.83  170.95  2098.4  175.77 2099.41   178.9 2099.82
  187.17 2100.49  214.33 2105.19
#Mann= 3 , 0 , 0
       0      .1       0   51.56     .05       0  109.34     .07       0
Bank Sta=51.56,109.34
Exp/Cntr=0.3,0.1

Type RM Length L Ch R = 1 ,377293.6,105.97,133.26,161.47
XS GIS Cut Line= 6
 1029916.7530746  656923.0141933 1029916.7530746  656954.6114194
 1029913.1072361  656975.2711303 1029916.7530746  656999.5766796
 1029919.1836234  657059.1252935 1029913.1072361  657084.6461323
#Sta/Elev= 28
       0 2109.34   29.31 2084.46    31.6 2082.65   32.56 2081.94   32.68 2081.88
    50.1  2079.2   52.58  2078.8   53.46  2078.6   54.27 2078.07   64.79 2071.09
    67.7 2069.21    74.3 2069.13   77.18 2069.89   78.54 2070.23   84.19 2070.74
   88.49 2071.17   91.78 2070.94   91.89 2070.94   97.19 2070.78  100.31 2070.74
   103.9 2070.72  112.19 2075.04  117.36 2077.74  119.65 2078.89  124.36 2080.18
  135.41 2085.41  136.96 2086.03  163.19 2097.14
#Mann= 3 , 0 , 0
       0      .1       0   64.79     .05       0   103.9     .07       0
Bank Sta=64.79,103.9
Exp/Cntr=0.3,0.1

Type RM Length L Ch R = 1 ,377160.3,114.95,106.93,95.32
XS GIS Cut Line= 6
 1029851.1280733  656912.0766779  1029821.961396  656943.6739041
 1029798.8711061   656974.055871 1029774.5655568  656995.9308714
 1029755.1211053  657015.3752926 1029751.4752971    657021.45168
#Sta/Elev= 20
       0 2122.62    1.63 2121.63   30.05 2095.05   57.84 2070.23   61.56 2069.11
   68.92 2066.27   74.44 2066.58   74.51 2066.58   75.27 2066.62   81.17 2066.85
   82.47 2066.88   93.08 2067.16   94.65 2067.16   97.83 2067.15   98.96  2067.8
   104.3 2070.47  115.82 2076.58  136.02 2089.28  141.37 2093.27  148.45 2098.53
#Mann= 3 , 0 , 0
       0      .1       0   61.56     .05       0   104.3     .07       0
Bank Sta=61.56,104.3
Exp/Cntr=0.3,0.1

Type RM Length L Ch R = 1 ,377053.4,319.56,327.43,341.87
XS GIS Cut Line= 6
 1029786.7183314  656847.6669663 1029733.2461049  656879.2641925
 1029719.8780709  656902.3544824 1029701.6489089  656924.2294828
 1029696.7877809  656940.0280959 1029684.6350063  656970.4100325
#Sta/Elev= 24
       0 2125.88    6.63 2122.91    9.51 2120.63   18.29  2113.2   22.81 2110.01
   27.78 2106.61   43.12 2093.91   44.63 2092.75   57.02 2085.07   62.11 2081.82
    67.3 2078.86   69.79 2076.63   78.31 2070.03   83.55 2067.17    89.9  2063.7
   90.61 2063.73  103.33 2062.78  117.38 2063.15  118.19 2063.76  124.51 2067.75
  164.06  2090.1  165.14 2091.15  165.74 2091.64  166.55 2091.84
#Mann= 3 , 0 , 0
       0      .1       0   83.55     .05       0  124.51     .07       0
Bank Sta=83.55,124.51
Exp/Cntr=0.3,0.1

Type RM Length L Ch R = 1 ,376726.0,510.53,463.05,440.68
XS GIS Cut Line= 3
 1029545.5972651  656644.8846522 1029482.5819689  656677.2925154
 1029405.1632015  656760.1126034
#Sta/Elev= 30
       0 2076.956.459991 2075.099.569992 2074.5413.76999 2075.54   17.69  2075.4
27.25999 2072.04   30.98 2070.1735.87999 2069.37   37.55 2069.22   42.97  2068.7
   46.58 2068.49   66.88 2062.7170.85999 2061.2779.32999 2058.84   82.02 2058.86
82.71999 2058.8883.89999 2058.91   91.12 2059.07   96.81 2059.32  100.82 2059.55
  102.31  2059.6  102.73 2059.68  102.86  2059.7  111.33 2060.92  114.79 2062.05
  115.77 2062.32  124.47 2062.66  129.25 2062.33  179.01 2087.96  184.23  2090.5
#Mann= 3 , 0 , 0
       0      .1       070.85999     .05       0  114.79     .07       0
Bank Sta=70.85999,114.79
Exp/Cntr=0.3,0.1

Type RM Length L Ch R = 1 ,376262.9,452.49,397.7,364.7
XS GIS Cut Line= 4
 1029066.6810383  656558.4636738  1029043.275356   656603.474578
 1029036.0736053  656666.4898742 1029028.8718546  656725.9043101
#Sta/Elev= 27
       0 2072.45    22.6 2063.48   30.33 2060.32   38.15 2056.89   47.75 2052.88
   50.73 2051.72   54.86 2050.06   56.77  2049.3   57.54 2049.18   59.41 2049.06
   68.99 2049.08   70.64 2048.84   74.89 2047.97   81.63 2046.59   86.07 2047.35
   90.61 2048.36   96.84 2048.55   98.02  2048.6   98.77 2048.69  108.81 2050.73
  112.07 2051.77  117.15 2055.27  133.33 2064.62  150.97 2076.35  163.22 2086.59
  173.85 2092.56  174.01 2092.66
#Mann= 3 , 0 , 0
       0      .1       0   68.99     .05       0   96.84     .07       0
Bank Sta=68.99,96.84
Exp/Cntr=0.3,0.1

Type RM Length L Ch R = 1 ,375865.2,333.12,360.33,364.57
XS GIS Cut Line= 6
 1028742.6023766   656264.992445 1028634.5761459  656297.4003082
 1028591.3656718   656448.637013 1028576.9621703  656576.4680354
 1028670.5848995  656704.2990579 1028699.3918722   656796.121357
#Sta/Elev= 30
       0 2087.3818.35004 2077.0925.29004 2073.69   42.06 2069.9356.54004 2068.81
  106.63 2068.98  125.57 2068.11  143.69 2065.79  152.87 2065.79  161.92 2064.17
  172.57 2062.86  208.85 2060.09  287.67 2058.25  309.71 2058.32  344.19 2057.81
  417.36 2056.26  460.34 2054.05  490.21 2051.42   509.7 2049.64  548.93 2043.57
  559.43 2044.94  562.59 2046.53  569.99 2048.72  577.92 2050.49  618.62 2055.65
   623.4  2056.7  626.44  2057.9  638.13  2064.7  650.42 2073.33  653.45 2074.92
#Mann= 4 ,-1 , 0
       0     .05       0  490.21     .08       0   509.7     .05       0
  577.92     .08       0
Bank Sta=509.7,577.92
Exp/Cntr=0.3,0.1

Type RM Length L Ch R = 1 ,375504.9,383.61,391.3,447.48
XS GIS Cut Line= 4
 1028168.2629602  656371.2182153 1028209.6730345  656432.4330814
 1028342.9053473  656860.9370833 1028387.9162818  656886.1431957
#Sta/Elev= 30
       0 2101.411.859985 2099.7114.96997 2091.0218.23999 2088.1725.95996  2082.7
47.73999 2065.7366.53998 2053.8467.09998 2053.75  156.48 2052.57  208.09 2052.81
     228 2052.33  256.48 2052.27  304.99 2053.22  347.72 2052.38  412.05  2049.5
  425.72 2047.97  440.06 2045.51   446.2 2044.88  456.92 2041.58  481.32 2040.65
     491 2046.77  496.04 2046.98  503.71 2050.15  512.98 2052.51  537.31 2053.66
  540.72 2054.68  545.74 2054.65  556.05 2055.36  559.75 2056.09  574.23 2061.18
#Mann= 4 ,-1 , 0
       0     .05       0  412.05     .08       0  425.72     .05       0
     491     .08       0
#XS Ineff= 2 , 0
       0     300    2060               0
Permanent Ineff=
       F       F
Bank Sta=425.72,491
Exp/Cntr=0.3,0.1

Type RM Length L Ch R = 1 ,375113.6,507.11,395.69,344.09
XS GIS Cut Line= 5
 1027885.5943727  656598.0732876 1027890.9956631  656670.0907647
 1027972.0153512  657001.3711771 1028094.4450531  657015.7746483
 1028144.8572779  657048.1825418
#Sta/Elev= 30
       0 2071.97    7.08 2069.44   27.66 2063.24   46.91 2057.03   75.38 2050.79
   86.04 2048.85  138.57 2048.69  164.75 2048.19  181.85 2048.14  188.44 2049.18
  196.99 2049.49  207.86 2049.04  217.78 2049.64  221.52 2049.62  274.61 2046.41
   293.7 2044.97  301.19 2043.52  342.94 2044.32   357.1 2046.86  359.56 2047.54
  373.89 2048.41  387.31 2048.85  400.26 2048.69  425.27 2049.07  473.81 2050.72
  493.54 2051.65  518.42 2053.29   535.8 2054.88  565.74 2058.76  596.47 2061.55
#Mann= 3 , 0 , 0
       0    .065       0  274.61     .05       0   357.1     .05       0
#XS Ineff= 2 , 0
       0  217.78 2049.64               0
Permanent Ineff=
       F       F
#Block Obstruct= 1 ,-1
  149.04  252.23 2059.98
Bank Sta=274.61,357.1
Exp/Cntr=0.3,0.1

Type RM Length L Ch R = 1 ,374717.9,445,383.1,136
XS GIS Cut Line= 6
  1027460.691231  656965.3624235  1027561.515711  657003.1716073
 1027703.7502349  657188.6166053 1027899.9978439  657206.6209973
 1028009.8245047  657251.6319015 1028031.4297569  657339.8533101
#Sta/Elev= 30
       0 2073.34    5.32 2069.88   22.88 2061.88   36.96 2055.87   57.87 2048.19
   63.11 2047.08   85.71 2046.06  103.95  2047.8  108.95  2047.5  119.55 2044.95
  125.17 2040.99  136.57 2037.91  151.05 2038.14  173.42 2042.17  186.03 2044.28
  274.97 2043.11  319.18 2046.49  440.16 2046.42  455.02 2047.05  482.98  2046.6
  545.77 2048.04  559.51 2048.78  611.27 2055.32  625.24 2054.19  654.58 2055.06
  659.59 2057.16  665.48 2058.31  674.25 2061.43  740.61 2065.21  750.42 2066.83
#Mann= 3 , 0 , 0
       0     .08       0  125.17     .05       0  173.42     .06       0
#XS Ineff= 2 , 0
       0                  186.03       0 2044.28
Permanent Ineff=
       F       F
Bank Sta=125.17,173.42
Exp/Cntr=0.3,0.1
