HEC-RAS study lds_broad_rvr.prj: Upper_Broad 3-06-07

--- lds_broad_rvr.g05 (geometry) --- (continued)

Type RM Length L Ch R = 1 ,374334.8,94,188.2,204.7
XS GIS Cut Line= 6
 1027232.7546536  657302.2603002 1027301.2276899  657322.8022081
  1027354.864877  657307.9663891 1027442.7385973  657217.8102211
 1027497.5170384  657209.8217148 1027950.8638765  657359.1242656
#Sta/Elev= 30
       0 2065.55    7.87 2063.05   20.91 2057.29   33.88 2050.25   53.32 2050.19
  117.72 2042.64  169.06 2039.15  179.77 2036.33  195.13  2036.1  198.91 2035.42
  208.28 2038.94  220.32 2043.46  261.82 2042.15  282.15  2044.8  291.33 2044.17
  383.01 2043.64  391.04 2044.26  418.12 2044.16  496.95 2045.59  619.94 2045.34
  653.39 2046.68  714.73 2047.82  745.56 2049.89  751.04 2051.63  757.63 2052.66
  764.26 2056.02   766.2 2057.78   777.1 2061.96   780.6 2061.64  785.89  2062.6
#Mann= 3 , 0 , 0
       0    .055       0  169.06     .05       0  208.28    .055       0
Bank Sta=169.06,208.28
Exp/Cntr=0.5,0.3

Type RM Length L Ch R = 1 ,374146.6,168,160.6,169
XS GIS Cut Line= 6
 1027198.5181506  657374.1569778 1027297.8040487  657412.9583458
 1027370.8419198  657425.5117474  1027483.822413  657428.9353886
 1027540.6479986   657424.108978 1027967.1100622  657371.3089124
#Sta/Elev= 30
       0 2070.54   12.86 2066.37      31 2056.89    46.4 2053.51   62.54 2048.16
    68.5 2047.11   88.09 2044.91   172.1 2040.08  259.47 2039.45  274.09 2038.26
  277.65 2037.18  280.46 2036.15  295.27 2035.41  304.13 2035.66  307.85  2037.3
  310.45 2038.44  333.87 2040.58  369.16 2042.28  468.96 2044.05  576.71 2044.39
  674.79 2047.11  683.74 2046.49  699.59 2047.85  707.96 2049.29  713.71 2048.93
  723.64 2055.97  727.23 2057.78  738.49 2059.63  742.45 2061.73   780.5 2064.18
#Mann= 3 , 0 , 0
       0    .055       0  277.65     .05       0  307.85    .055       0
#XS Ineff= 2 , 0
       0  208.75    2052  374.75       0    2052
Permanent Ineff=
       F       F
Bank Sta=277.65,307.85
Exp/Cntr=0.5,0.3

Type RM Length L Ch R = 3 ,374070. ,,,
BEGIN DESCRIPTION:
STR_149
END DESCRIPTION:
Bridge Culvert--1,0,-1,-1, 0
Deck Dist Width WeirC Skew NumUp NumDn MinLoCord MaxHiCord MaxSubmerge Is_Ogee
120,30,2.6,0, 7, 7, , , 0.95, 0, 0,0,,
       0  228.75  228.75  354.75  354.75  475.64  742.45
    2054    2052    2052    2052    2052    2054 2061.73
                    2049    2049
       0   118.7   118.7   244.7   244.7  362.88  514.19
    2054    2052    2052    2052    2052    2054 2053.99
                    2049    2049
Pier Skew, UpSta & Num, DnSta & Num=  ,270.75, 2 ,160.7, 2 , 0 , 0 , 0 ,,
       2       2
    2030    2049
       2       2
    2030    2049
Pier Skew, UpSta & Num, DnSta & Num=  ,312.75, 2 ,202.7, 2 , 0 , 0 , 0 ,,
       2       2
    2030    2049
       2       2
    2030    2049
BR Coef=-1 , 1 , 0 ,, 0 ,,,0.8,0,2,0,
WSPro=,,,, 1 ,,,, 0 ,,,, 0 ,,,,-1 ,-1 ,-1 , 0 , 0 , 0 , 0 , 0
BC Design=,, 0 ,, 0 ,,,,,,

Type RM Length L Ch R = 1 ,373986.0,72,117.2,112
XS GIS Cut Line= 6
 1027253.2965615  657572.7287437 1027437.0325387  657586.4233691
 1027466.7041766  657587.5645627 1027519.2001701  657594.4118754
 1027624.5865489  657585.2168573 1027764.0328775  657612.2938334
#Sta/Elev= 30
       0 2044.63    9.69 2044.92   15.15 2044.66   27.53 2040.55   31.46 2039.61
   45.49 2038.57   57.21 2038.16   85.57 2038.53  134.73 2038.57  157.09 2037.02
  163.42 2035.38  198.79  2035.8  209.74 2035.58   213.3 2035.75  218.922036.924
  227.83 2038.87  234.64 2039.78  254.24  2040.5  273.19 2040.79  286.73 2040.57
   314.8 2037.94  321.77 2038.63  337.83  2039.2  366.73 2041.15  409.16 2042.61
  455.31 2046.43  471.88 2049.12  493.32 2051.05  509.53  2053.6  514.72 2054.02
#Mann= 3 , 0 , 0
       0    .055       0  157.09     .05       0  218.92    .055       0
#XS Ineff= 2 , 0
       0    88.7    2044   274.7       0    2044
Permanent Ineff=
       F       F
Bank Sta=157.09,218.92
Exp/Cntr=0.5,0.3

Type RM Length L Ch R = 1 ,373868.8,121.83,311.07,480.7
XS GIS Cut Line= 6
 1027229.3410008  657525.7759974 1027225.2230424  657566.9555204
 1027235.7051155  657627.9760964 1027426.7615847  657702.8275036
 1027455.2919989  657706.2511448 1027734.2482189  657690.8169884
#Sta/Elev= 30
       0 2052.96    2.56 2053.15   15.72 2044.65   25.79 2041.37   31.34 2040.96
   95.03  2040.6  118.02 2039.15  123.76 2038.19   149.7 2037.09  218.74  2037.6
  251.79 2039.44  260.06 2038.72  267.82    2039  273.41 2037.73  280.96 2036.85
  287.65 2034.93  291.38 2034.65  314.56 2033.69  322.14 2032.55  328.89 2033.82
  340.63 2039.64  342.62 2039.93  349.21 2039.53  355.29 2040.11  473.89 2039.59
  497.82 2037.03  542.34 2044.61   564.1    2047   581.6 2049.82   616.8 2053.55
#Mann= 3 , 0 , 0
       0    .065       0  291.38     .05       0  328.89    .065       0
Bank Sta=291.38,328.89
Exp/Cntr=0.3,0.1

Type RM Length L Ch R = 1 ,373557.9,127.65,410.93,509.09
XS GIS Cut Line= 6
 1027208.2165252  657544.6952389 1027222.9857243  657612.2116255
 1027174.4583167  657705.0466609 1027218.7659445  657935.0243291
 1027303.1614202  657960.3429779 1027332.6998488  658127.0240696
#Sta/Elev= 30
       0 2043.01 7.72998 2041.4322.15997 2040.27  175.98 2040.46  190.34 2039.38
  221.45 2038.67  265.61 2035.56  370.34  2036.3  387.87 2037.34  403.26 2033.89
  420.77 2034.98  431.76 2034.09  459.33 2033.43  466.24  2034.8  473.92 2035.37
  481.55 2037.59  489.39 2036.74   513.5 2037.64  540.18  2037.3  558.32 2038.22
  570.29 2040.06  583.82 2036.93  598.91 2038.69  606.49 2038.36   617.8 2043.13
  635.85 2053.21  642.91 2053.38  650.96 2054.69   662.8 2058.31  669.06 2063.82
#Mann= 3 , 0 , 0
       0     .05       0  420.77     .05       0  473.92     .08       0
#XS Ineff= 4 ,-1
     210  387.87 2037.34     395  420.77 2034.98  481.55  558.89 2037.59
  570.29     640 2040.06
Permanent Ineff=
       T       F       F       F
Bank Sta=420.77,473.92
Exp/Cntr=0.3,0.1

Type RM Length L Ch R = 1 ,373146.9,428.53,472.99,488.71
XS GIS Cut Line= 6
 1027180.7879865   657618.541265 1027119.6012394  657650.1895836
 1026982.4585762  657730.3652794  1026950.810288  657802.1014458
 1026872.7444518  657909.7057106 1026693.4040508  657854.8486333
#Sta/Elev= 30
       0 2040.2716.09003 2040.6633.14001 2039.54  192.82 2036.56  237.36 2034.75
  245.87 2033.61  284.35 2031.09  297.28 2030.55  321.79 2028.17  336.89 2028.06
  349.56 2031.24  351.79 2031.24  366.15 2030.52  398.96 2033.61  444.08 2034.81
  446.69 2034.55  463.01 2029.47  464.64 2028.31  469.76 2028.97  482.24 2032.77
  493.75    2035  504.24 2039.21  524.58 2054.28  531.82 2058.49  539.77 2061.15
  557.38 2061.65  570.71 2064.15  583.74 2078.97  612.92 2091.87  626.64  2095.9
#Mann= 4 ,-1 , 0
       0     .05       0  284.35     .08       0  297.28     .05       0
  351.79     .08       0
#XS Ineff= 2 , 0
       0                  444.08       0 2034.81
Permanent Ineff=
       F       F
Bank Sta=297.28,351.79
Exp/Cntr=0.3,0.1

Type RM Length L Ch R = 1 ,372673.9,371.64,364.59,371.31
XS GIS Cut Line= 6
 1026797.7954606  657385.9391815 1026772.3961477  657428.7169446
 1026741.6496333  657452.7794421 1026712.2399041   657471.494738
 1026664.1149093  657492.8836044 1026587.9169705  657541.0086295
#Sta/Elev= 30
       0 2055.16    6.61 2055.78      13 2053.82   21.01 2052.67   25.82 2049.91
   33.31 2047.04   45.43 2041.09   48.46 2040.12      59 2038.73   61.16 2038.53
   70.73 2037.34   79.57 2036.86   86.22 2036.31  108.71 2030.08  110.32 2029.75
  129.84 2024.86  139.29 2024.81  158.06 2024.81  170.58 2025.01  179.96 2028.15
  196.06 2033.01  220.43 2042.92  229.35 2046.02  240.06 2050.21  241.76 2051.13
  248.78 2051.09  250.42 2051.45  262.08  2054.6  262.71 2054.91  266.74 2057.72
#Mann= 3 , 0 , 0
       0     .08       0  110.32     .05       0  179.96     .06       0
Bank Sta=110.32,179.96
Exp/Cntr=0.3,0.1

Type RM Length L Ch R = 1 ,372309.3,249.18,248.54,208.07
XS GIS Cut Line= 6
 1026551.8232244  657115.9044479   1026521.07671  657158.6822413
 1026462.2572517  657193.4391719 1026428.8371063  657204.1336051
 1026395.4169912  657236.2169653 1026386.0593432  657252.2586302
#Sta/Elev= 28
       0 2053.17   12.51 2054.06   14.89 2054.39   31.78 2046.99   36.36 2045.34
   44.42 2041.25   66.19 2022.89   67.66 2021.29   76.96 2021.05   89.62 2021.11
   95.49 2021.47  100.76 2021.31  110.83 2025.78  112.21 2026.18   112.8 2026.24
  121.13 2026.87  126.96 2027.16  137.69 2030.19  139.72 2030.42  161.74    2032
  169.82 2032.95  174.07 2033.66  179.42 2034.63  191.79  2038.3  196.55 2039.79
  203.76 2042.42  214.89 2044.05  222.33 2044.88
#Mann= 3 , 0 , 0
       0    .065       0   66.19     .05       0  110.83    .065       0
Bank Sta=66.19,110.83
Exp/Cntr=0.3,0.1

Type RM Length L Ch R = 1 ,372060.8,235.44,207.03,155.83
XS GIS Cut Line= 6
 1026472.9517152  656942.1197343 1026408.7850251  656940.7829188
 1026343.2815498  656971.5294634 1026335.2607174  656983.5607121
 1026320.5558679  657025.0016597 1026268.4204568  657069.1162686
#Sta/Elev= 30
       0 2050.35    5.81 2050.14   16.33 2049.41   24.41 2048.51   41.83 2049.95
   64.29 2032.64   76.09 2026.72   82.12 2024.61   90.15 2021.71   92.43  2019.7
   97.19 2019.56     103 2019.61  118.22 2019.49   126.8 2019.61     134 2021.54
  151.35 2024.86  152.53 2025.08  154.34 2025.06  159.84 2025.41   171.6 2026.69
  175.17 2027.24  181.64 2028.07  188.45 2028.33  201.16 2029.41  214.44 2030.26
   227.8 2031.25  234.78 2032.21  239.03 2032.88  250.96 2035.66  263.66 2039.97
#Mann= 3 , 0 , 0
       0    .065       0   82.12     .05       0  151.35    .065       0
Bank Sta=82.12,151.35
Exp/Cntr=0.3,0.1

Type RM Length L Ch R = 1 ,371853.8,195.38,184.79,124.41
XS GIS Cut Line= 6
 1026289.8093535  656670.7482154 1026287.1357225  656718.8732102
 1026225.6426635  656832.5016804 1026228.3162945  656879.2898597
 1026206.9273978  656902.0155719 1026178.8544841  657016.9808272
#Sta/Elev= 30
       0 2064.52    2.18 2062.68    8.08 2060.16   33.29 2053.02   40.42 2048.62
   48.12 2045.52   60.99 2044.98   73.34 2043.87    79.1 2043.25   87.54  2041.6
   91.07  2040.1   95.23 2035.92  106.67 2026.79  115.59 2020.94  122.44  2017.4
  125.55 2017.82  140.77 2016.91   165.3 2021.29  180.46 2024.69  195.36 2024.85
  225.13 2022.96  232.36 2022.99  237.23 2023.23  256.22  2028.2  281.67 2028.54
  340.85 2031.92  354.36 2033.89  360.88 2036.74  367.68 2040.39  377.61 2040.56
#Mann= 3 , 0 , 0
       0      .1       0  115.59     .05       0   165.3     .08       0
#XS Ineff= 2 , 0
       0                  195.36       0 2024.85
Permanent Ineff=
       F       F
Bank Sta=115.59,165.3
Exp/Cntr=0.3,0.1

Type RM Length L Ch R = 1 ,371669.0,228.39,218.82,187.22
XS GIS Cut Line= 6
 1026074.5836317  656689.4634811  1026065.226014   656792.397518
 1026087.9516959  656872.6058427 1026086.6149107  656887.3106922
 1026067.8996148  656912.7100051 1026050.5211343  656960.8349999
#Sta/Elev= 30
       0 2041.05   19.84 2040.36   33.21 2039.14   42.32 2037.28   46.76 2036.66
   55.26 2029.44   62.06 2024.64   72.51 2019.66   77.89 2017.93   82.73    2017
   87.52 2017.24   99.69 2016.74  106.49 2018.35  123.53  2020.3  131.08 2021.74
  155.39 2023.46  175.09 2025.95  204.52 2027.73   205.3 2028.05  218.56 2030.48
  224.59 2030.55  229.77  2032.3  234.82 2033.28  247.67 2037.03  248.96 2037.57
  262.37 2038.93  271.42 2039.46  275.95 2039.44  281.91 2041.35  286.04 2042.22
#Mann= 3 , 0 , 0
       0      .1       0   77.89     .05       0  106.49     .08       0
Bank Sta=77.89,106.49
Exp/Cntr=0.3,0.1

Type RM Length L Ch R = 1 ,371450.2,148.31,105.89,91.13
XS GIS Cut Line= 6
 1025826.1234283  656696.2863373 1025850.0438781  656806.9184895
 1025852.2864326  656821.1212537 1025859.0140657  656833.0814937
 1025891.9047031  656851.0218387 1025918.8152053  656904.8428734
#Sta/Elev= 30
       0 2057.15     .32 2057.07    5.83 2053.56   34.03 2036.75   37.59 2036.69
    56.1 2036.77   77.96 2036.16   83.98 2036.41   94.99 2027.71  101.25 2022.19
  110.96 2018.17  112.21 2017.77  112.63 2017.85  117.65 2016.72  122.17  2015.7
  127.57 2015.36  136.11  2015.1  142.95 2015.43  148.67  2015.5  154.68 2015.86
  178.76 2019.85   186.3 2020.86  209.96  2028.1   213.5 2029.56  218.17  2030.2
   220.9 2031.17  226.49 2033.55  229.14 2033.95  234.05 2035.32  238.94 2035.46
#Mann= 3 , 0 , 0
       0     .07       0  117.65     .05       0  154.68     .07       0
Bank Sta=117.65,154.68
Exp/Cntr=0.5,0.3

Type RM Length L Ch R = 1 ,371344.3,16.13,21.57,17.89
XS GIS Cut Line= 6
 1025657.9326607  656732.1670271 1025679.6105863  656747.8648478
 1025686.3382194   656804.675935  1025811.810186  656889.0385397
 1025833.3396774  656941.6105663 1025833.8403703  656984.6695795
#Sta/Elev= 30
       0    2053   14.74 2047.32   26.76  2043.5   30.72 2041.08   38.06 2037.59
   40.33    2036   51.39 2034.32   72.99 2034.05   95.23 2032.38  101.42 2032.34
  103.98 2030.67  115.78 2016.91  124.42 2014.61   139.8 2011.38  156.35 2010.14
  169.36 2011.29  189.42 2011.99  209.39 2013.08  215.76 2012.73  226.25 2014.85
  232.31 2018.63  235.75 2019.33  250.14 2026.55  258.18 2031.58  280.07 2031.68
  296.57 2032.67  305.11 2035.38  311.33    2038  326.12 2042.33  335.62 2046.66
#Mann= 3 , 0 , 0
       0     .07       0   139.8     .05       0  189.42     .07       0
Bank Sta=139.8,189.42
Exp/Cntr=0.5,0.3

Type RM Length L Ch R = 3 ,371333.5,,,
BEGIN DESCRIPTION:
STR_147
END DESCRIPTION:
Bridge Culvert--1,0,-1,-1, 0
Deck Dist Width WeirC Skew NumUp NumDn MinLoCord MaxHiCord MaxSubmerge Is_Ogee
4.5,12,2.6,0, 2, 2, 2031, , 0.95, 0, 0,0,,
      80     270
    2032    2031
  2028.5  2027.5
      50     309
    2032    2031
  2028.5  2027.5
BR Coef=-1 , 1 , 0 ,, 0 ,,,0.8,0,2,0,
WSPro=,,,, 1 ,,,, 0 ,,,, 0 ,,,,-1 ,-1 ,-1 , 0 , 0 , 0 , 0 , 0
BC Design=,, 0 ,, 0 ,,,,,,

Type RM Length L Ch R = 1 ,371322.7,139.27,169.74,232.9
XS GIS Cut Line= 6
 1025630.0611199  656741.8368287 1025642.0775978  656806.9260262
 1025676.6205338  656818.8786992 1025793.7854842  656898.0508906
 1025811.3094931  656959.1346055 1025810.8088304   656988.675062
#Sta/Elev= 30
       0 2054.02    6.53  2050.6    32.5 2033.16   52.93 2033.73   77.35 2033.37
   78.96 2033.09   89.95 2033.17  104.47 2032.62  112.56 2031.43  134.07 2015.65
  134.66 2014.96  141.67 2012.48  143.59 2012.26  153.66 2010.95  187.49 2010.67
  202.31 2010.74   211.4 2011.65  227.64 2013.31  236.15 2014.85  244.61 2020.58
  251.87 2026.09  257.57 2029.35  259.11 2029.64  265.53 2028.82  284.67 2030.03
  306.29 2030.84  318.28 2037.63  324.22 2040.64  333.21 2043.85  338.52 2046.18
#Mann= 3 , 0 , 0
       0     .07       0  143.59     .05       0   211.4     .07       0
#XS Ineff= 1 ,-1
  250.28  309.64    2031
Permanent Ineff=
       F
Bank Sta=143.59,211.4
Exp/Cntr=0.5,0.3

Type RM Length L Ch R = 1 ,371153.0,548.38,608.93,597.08
XS GIS Cut Line= 5
 1025547.2765362  656732.5939267 1025551.8604701  656854.8317598
 1025573.2520909  656917.4786342 1025580.8919403  657013.7409127
 1025574.7800487  657068.7479376
#Sta/Elev= 30
       0 2060.35   22.15 2046.06   42.85 2031.61   64.01 2032.51   76.98 2032.58
   85.91 2032.29  109.16 2031.01  113.59 2030.53   123.5 2028.95  127.38 2026.15
  140.12 2018.19  148.85 2010.62  154.93 2009.62  184.98 2009.97   197.9 2010.69
  215.81 2013.43  226.91 2015.47  244.55 2022.11  247.67 2023.61  256.78 2025.95
  282.04 2027.54  283.29 2027.37  285.09 2027.49  292.25 2028.37   298.8  2032.8
  303.06 2034.74  314.12 2036.74  328.64 2040.43   335.3 2042.61  340.43 2044.81
#Mann= 3 , 0 , 0
       0    .065       0  148.85     .05       0   197.9     .07       0
Bank Sta=148.85,197.9
Exp/Cntr=0.3,0.1

Type RM Length L Ch R = 1 ,370544.0,441.22,473.63,487.56
XS GIS Cut Line= 5
 1025198.8987722  656561.4609905 1025020.1259564  656778.4331141
 1025009.4301611  657168.0661619 1025043.0455652  657242.9368195
 1025049.1574569  657293.3599106
#Sta/Elev= 30
       0 2038.067.800049 2035.0526.21002 2029.9757.62006 2022.4189.73004 2026.06
  100.55 2024.84  110.01 2021.16120.4301  2019.5  156.97 2017.87  281.02 2016.02
  354.49 2016.02  397.18 2016.73  452.28 2015.81  472.66 2014.45  495.65 2011.05
  508.34    2010     541 2009.05  553.26 2008.46565.9901 2004.87589.1801 2004.28
  602.59 2004.29  607.57 2007.12  619.53 2013.36  629.97  2015.4  651.92 2015.29
  663.48    2018  676.87 2019.87  712.25 2022.89751.2401 2028.13  803.78 2064.26
#Mann= 5 ,-1 , 0
       0     .05       0     541     .08       0  553.26     .05       0
  607.57     .08       0  619.53     .05       0
Bank Sta=553.26,607.57
Exp/Cntr=0.3,0.1

Type RM Length L Ch R = 1 ,370070.4,456.46,499.62,611.98
XS GIS Cut Line= 6
 1024900.9440993   656414.775621 1024841.3531405  656559.9330025
 1024696.1957591  656677.5869017 1024545.2236267  657057.7472227
 1024534.0448453   657165.808988 1024536.0632351  657329.6094763
#Sta/Elev= 30
       0 2041.09      40 2030.9653.10999 2026.0766.22998 2020.2278.72998  2020.1
  172.37 2014.69  240.57 2014.75  343.81 2011.16  516.28 2013.27  610.23 2011.41
  665.48 2012.06  706.64  2013.5  732.67 2013.02742.5699 2008.64  751.34 2005.68
  762.92 2004.88  789.38 2004.72  800.78 2002.92   812.2 2003.53  823.44 2006.61
  828.39 2008.41  859.87 2008.36  874.41 2012.53  911.02 2013.19  946.97 2015.92
  968.72 2021.35  986.75 2028.83  994.76 2034.74 1010.65 2042.82 1025.48 2047.02
#Mann= 4 ,-1 , 0
       0     .05       0  732.67     .08       0  751.34     .05       0
  823.44     .05       0
#XS Ineff= 2 , 0
       0                  846.03       0 2008.79
Permanent Ineff=
       F       F
Bank Sta=751.34,823.44
Exp/Cntr=0.3,0.1

Type RM Length L Ch R = 1 ,369570.8,122.89,495.14,576.87
XS GIS Cut Line= 6
 1024497.2479438   656543.988074  1024472.406167  656666.6443922
 1024289.1980028  656722.5384202 1024099.7794246  656956.9827339
 1024011.2805495  657017.5345799 1023933.6499971  657023.7450241
#Sta/Elev= 30
       0 2023.249.820007 2016.3524.14001 2010.17   53.06 2008.24   67.56 2007.99
  125.14 2009.45  181.21 2008.77  208.69 2007.55  242.95 2004.78  259.85 2004.33
  358.86 2003.86  390.69 2004.29  410.99 2003.77   432.6 2004.42   446.5 2005.52
  490.87 2006.05  547.71 2005.52  592.35 2006.13  603.22  2007.1  608.12 2007.04
  618.09 2005.15  625.09 2003.87  648.79 2001.22  659.41 2000.96  673.56  2005.1
  709.58 2015.63  719.46 2019.27  757.66 2030.97  773.62 2035.11   803.2  2046.1
#Mann= 3 , 0 , 0
       0     .08       0  618.09     .05       0  673.56    .065       0
#XS Ineff= 2 , 0
   803.2  199.98  2007.1           803.2
Permanent Ineff=
       F       F
Bank Sta=618.09,673.56
Exp/Cntr=0.3,0.1

Type RM Length L Ch R = 1 ,369075.6,69.55,175.31,151.75
XS GIS Cut Line= 5
 1024442.7716678   656536.719764 1024418.7297224   656579.995284
 1024316.5514163  656629.2812676 1024257.6486303    656682.17359
 1024165.0870964  656576.3889755
#Sta/Elev= 30
       0 2015.19   10.31 2012.82   16.77 2011.46   29.86 2009.06      43 2007.56
   49.51 2007.18   74.64 2006.09   89.47 2005.78   99.92 2005.37  109.42 2004.93
  128.35 2003.71  139.99 2003.14  162.95 2002.95  176.32 2003.02  201.13 2002.83
  225.59  2002.8  231.03  2003.3  235.62 2003.45  247.53 2003.04  255.71 2003.01
  260.82 2002.74  287.33 1999.32  313.25 1996.79  327.42  1997.2  338.75 1997.35
  339.59 1997.28  340.37 1997.58  352.31 1999.31  369.45 2004.87  382.68 2008.87
#Mann= 3 , 0 , 0
       0    .065       0  287.33     .05       0  352.31     .08       0
Bank Sta=287.33,352.31
Exp/Cntr=0.3,0.1

Type RM Length L Ch R = 1 ,368900.3,423.87,433.79,462.21
XS GIS Cut Line= 4
 1024536.0632351    656478.77841 1024391.6703622  656530.0145897
 1024272.1192964  656460.1470774 1024151.0156043  656444.6209669
#Sta/Elev= 30
       0 2031.36   10.57 2031.13   15.29 2031.95   21.09 2031.58   48.86 2028.26
   66.75 2027.49   73.07 2026.61   99.25 2020.81  107.89 2018.37  111.34 2018.21
  121.83 2015.19  125.77 2015.05  134.36 2012.12  143.96 2012.28  153.21 2010.55
  159.74 2010.16  166.66 2008.97  173.95 2005.95  188.55 2003.45  206.14 1999.34
  229.94 1995.39  245.91 1995.26  253.17 1995.43  257.31 1998.39  261.99 2001.09
  284.35 2002.53  307.98 2005.08  347.16  2010.5  376.46 2022.08  413.78 2042.52
#Mann= 3 , 0 , 0
       0     .08       0  206.14     .05       0  257.31     .08       0
Bank Sta=206.14,257.31
Exp/Cntr=0.3,0.1

Type RM Length L Ch R = 1 ,368466.5,357.6,353.23,339.84
XS GIS Cut Line= 4
 1024904.0321595  656373.2008284 1024792.2441337  656241.2288439
 1024596.6150811  656168.2561095  1024442.906542  656033.1789332
#Sta/Elev= 30
       0 2043.8114.52002 2040.8531.08002 2035.6940.91998 2031.5655.48999 2027.38
65.82001  2023.873.97003 2012.83   78.28 2011.13   98.37 2008.63  139.56 2005.69
  268.92 2002.68  316.93 2003.72  337.73 2003.58  383.56 2004.37   406.3 1999.71
  421.01 1995.73  427.48 1994.81   435.6 1991.06  442.03 1991.57  457.06  1991.5
  462.84 1992.42   467.7 1994.44  480.23 1999.64  486.42 2001.73  509.44 2004.97
   546.2 2013.27  554.86 2014.84   561.9 2017.61  568.79 2019.67  586.38 2026.64
#Mann= 4 ,-1 , 0
       0     .05       0   406.3     .08       0  427.48     .05       0
   467.7      .1       0
Bank Sta=427.48,467.7
Exp/Cntr=0.3,0.1

Type RM Length L Ch R = 1 ,368113.3,219.7,229.95,250.97
XS GIS Cut Line= 6
 1025259.6377954  656304.1490381 1024772.9092826  655854.0074578
 1024758.7255872  655848.3339978 1024724.6847363  655846.9156101
 1024710.5010409  655844.0788952 1024696.3173758  655831.3135572
#Sta/Elev= 30
       0 2022.86   46.54 2008.25   92.37 2004.97  146.88 2002.61  164.28 2002.32
  199.54 2002.91  214.95 2004.64   246.3 2010.81  267.71 2011.88   272.7 2010.38
  286.48 2003.19  317.93 2002.06  388.82 2001.97  426.69 2000.74   461.4 1998.26
  475.39 1998.67   501.8 2000.77  567.73 2001.43  576.62 2000.93  582.89 1999.85
  597.83 1995.54  605.76 1990.58  627.07 1990.11  638.85 1990.44  653.96 1994.08
  661.39 1999.59  666.46 2002.49  707.18 2005.72  720.91 2007.98  745.87 2018.93
#Mann= 3 , 0 , 0
       0    .055       0  597.83     .05       0  653.96      .1       0
#Block Obstruct= 1 ,-1
  334.27  498.34 2009.97
Bank Sta=597.83,653.96
Exp/Cntr=0.5,0.3

Type RM Length L Ch R = 1 ,367883.4,43.65,30.51,56.92
XS GIS Cut Line= 6
 1025406.1723699  656156.7616028   1025048.28471  655819.9825885
 1024950.4173207  655701.9660183 1024864.0637187  655621.3693554
 1024768.1152889  655579.1520342 1024745.0876839  655546.5295711
#Sta/Elev= 30
       0 2024.8829.90002  2011.1  106.86  2004.2   149.8 2002.64  233.78 2001.87
  248.47 2002.25  269.87 2004.46  300.68 2005.61  340.77 2001.59  429.11 1999.27
  439.13  1998.4  503.36  1995.7  549.55 1995.39  572.47 1993.41  585.92 1991.33
  621.65 1990.84  627.34 1989.99  631.18  1990.2  638.03 1993.16  640.97 1993.19
  676.67 1997.42  736.52 2001.39  762.01 2002.02  804.96  2004.1     845 2007.28
  858.45 2008.97   869.6 2011.35  888.77 2017.79  901.35 2023.26  907.63 2027.09
#Mann= 3 , 0 , 0
       0    .055       0  572.47     .05       0  640.97      .1       0
#XS Ineff= 2 ,-1
  549.89  568.37    1995   642.7  657.43    1995
Permanent Ineff=
       T       T
#Block Obstruct= 1 ,-1
  357.96  523.57 2011.54
Bank Sta=572.47,640.97
Exp/Cntr=0.5,0.3

Type RM Length L Ch R = 3 ,367868. ,,,
BEGIN DESCRIPTION:
Private_1
END DESCRIPTION:
Bridge Culvert--1,0,-1,-1, 0
Deck Dist Width WeirC Skew NumUp NumDn MinLoCord MaxHiCord MaxSubmerge Is_Ogee
7,16,2.6,0, 2, 2, 1994, , 0.95, 0, 0,0,,
     400     700
    1995    1995
  1993.5  1993.5
     400     700
    1995    1995
  1993.5  1993.5
BR Coef=-1 , 1 , 0 ,, 0 ,,,0.8,0,2,0,
WSPro=,,,, 1 ,,,, 0 ,,,, 0 ,,,,-1 ,-1 ,-1 , 0 , 0 , 0 , 0 , 0
BC Design=,, 0 ,, 0 ,,,,,,

Type RM Length L Ch R = 1 ,367852.9,197.68,198.25,169.86
XS GIS Cut Line= 6
 1025382.8568862  656088.1584748 1024974.1165721  655687.0940291
 1024958.7648355  655635.2818497 1024882.9655562  655553.7256919
 1024811.0042566  655542.2118743 1024790.8550757  655506.7109568
#Sta/Elev= 30
       0 2007.994.409973 2007.0632.98999 2004.7766.59998  2003.1  192.62 2000.92
  217.47 2004.14   237.4 2005.33  248.43 2002.84   254.6 2000.64  345.74 1999.53
  385.61 1996.54  482.65 1993.91  488.39 1994.22  494.17 1993.66  497.48 1992.63
  501.75 1991.58  528.72 1989.16  545.75  1990.3553.0599 1989.42   572.2 1992.86
  619.43 1998.68   637.3  2000.2  663.49 2001.05   735.9 2001.65  771.29 2002.82
  785.65  2003.6  815.41  2006.9  817.79 2007.69  829.24 2014.43  851.72 2029.22
#Mann= 3 , 0 , 0
       0    .055       0  497.48     .05       0   572.2      .1       0
#XS Ineff= 2 ,-1
  451.22  496.67    1995  572.06  595.34    1995
Permanent Ineff=
       T       T
#Block Obstruct= 1 ,-1
  292.99  433.12 2012.78
Bank Sta=497.48,572.2
Exp/Cntr=0.5,0.3

Type RM Length L Ch R = 1 ,367654.6,428.3,445.59,420.41
XS GIS Cut Line= 6
 1025538.2933636   655886.666757  1025388.613795  655809.9080132
  1025279.232588  655713.9595834 1025103.3891373  655530.6194205
 1024989.9196649  655442.6805634 1024923.2563509  655407.2213552
#Sta/Elev= 30
       0 2011.25    9.48 2009.34   41.98 2005.42   71.09 2003.19  114.84 2001.05
   165.5 2000.16  178.81 2003.59  200.01  2003.8  217.19  2003.4  227.52 2001.91
  243.57 2001.24  249.46 2000.11  310.44 1998.03  350.84 1995.12  397.63 1994.69
  403.67 1994.89  413.61 1996.29  429.19 1995.04  441.74 1993.66  466.59    1989
   476.4 1989.15  499.04 1993.57  506.44 1994.72  512.55 1996.63  524.01 1998.46
  566.91 2000.05  675.77 1999.98  732.06 2000.57  759.85 2001.06     787 2003.02
#Mann= 5 ,-1 , 0
       0     .05       0  429.19     .08       0  441.74     .05       0
  499.04     .08       0  512.55     .05       0
Bank Sta=441.74,499.04
Exp/Cntr=0.3,0.1

Type RM Length L Ch R = 1 ,367209.0,588.58,509.29,399.04
XS GIS Cut Line= 4
  1025713.299935  655542.5173387 1025558.6955243  655416.0228291
  1025500.133253  655305.9257542 1025118.3071944  655062.3067019
#Sta/Elev= 30
       0 2019.1210.35004 2014.0915.65002 2013.74   25.25  2010.132.29004  2008.3
94.95001 2003.13  135.11 1996.43  152.57 1995.03  169.81 1992.76  235.58 1992.99
  252.54 1992.42  262.12 1991.28  275.94 1988.34  300.75 1986.02  306.22 1986.64
  312.77 1988.43   316.4 1990.95  323.69 1996.06  325.03 1996.29  329.97 1995.39
  377.78 1997.46  426.01 1996.77  501.26 1997.43   610.7 1996.55  667.73  1997.9
   713.9 2001.75  723.47 2003.07  745.01 2009.43  760.63 2015.48  777.39 2023.76
#Mann= 5 ,-1 , 0
       0     .05       0  252.54     .08       0  262.12     .05       0
   316.4     .08       0  325.03     .05       0
Bank Sta=262.12,316.4
Exp/Cntr=0.3,0.1

Type RM Length L Ch R = 1 ,366699.7,561.8,544.41,532.69
XS GIS Cut Line= 5
 1026067.0160622  655038.8817692 1025992.0563562  655001.4019313
 1025938.1790532  654985.0044965 1025427.5160159  654903.0172925
 1025352.5563099  654865.5374546
#Sta/Elev= 30
       0 2051.1419.66998 2041.0873.84998 2015.6975.65002  2014.289.65002 2008.26
  101.58 2006.25  120.04  2005.8  124.49  2003.4     131 2001.46  138.48 1995.77
  155.13  1986.6  169.11 1985.98  176.79  1984.8  196.12 1989.05  215.05  1984.4
   233.8 1984.71  244.71 1985.68  253.24 1990.24  261.45 1990.25   299.9 1989.95
  318.38 1994.35  336.27 1995.03  635.27 1994.29  653.17 1995.07  678.62 1999.36
  694.09 2006.14  705.94 2012.41  725.97 2024.64  733.08 2027.44  741.13  2033.1
#Mann= 5 ,-1 , 0
       0    .065       0  176.79     .08       0  196.12     .05       0
  253.24     .08       0  261.45     .05       0
#XS Ineff= 2 , 0
       0  196.12 1989.05  253.55       0 1990.34
Permanent Ineff=
       F       F
Bank Sta=196.12,253.24
Exp/Cntr=0.3,0.1

Type RM Length L Ch R = 1 ,366155.3,571.38,519.44,541.6
XS GIS Cut Line= 6
 1026177.1131371  654600.8359689 1026111.5233981  654577.4110664
  1026017.823758  654467.3139915 1025956.9189873  654436.8615911
 1025624.2852633  654420.4641563 1025551.6680565  654380.6418191
#Sta/Elev= 30
       0 2010.2116.80005 2005.3238.48004  2001.563.72003 2003.2280.42004 1998.87
96.85004 1996.57  162.75 1993.56  195.54 1992.88  204.88 1993.21  212.62 1992.09
   224.9 1988.61  228.77 1987.97  237.36 1987.07  270.79 1986.26  282.73 1984.88
  308.06  1981.8  316.16 1981.68  329.25    1982  338.62 1984.24  346.12 1986.44
  374.96 1986.39     433 1991.15  480.26 1991.52  506.54 1990.68  582.32 1990.25
608.3101 1990.98  624.91 1992.62  671.08 2024.32  674.83 2027.53  698.59 2045.53
#Mann= 3 , 0 , 0
       0     .05       0  282.73     .05       0  338.62     .05       0
#XS Ineff= 2 , 0
       0                  351.77       0 1986.45
Permanent Ineff=
       F       F
Bank Sta=282.73,338.62
Exp/Cntr=0.3,0.1

Type RM Length L Ch R = 1 ,365635.9,769.5,399.69,269.19
XS GIS Cut Line= 6
 1026441.8146228  654247.1198114  1026416.047221  654174.5026047
 1026308.2926454   654104.227867  1026158.373203  653940.2534892
 1025781.2321734  653898.0886527 1025643.0251974  653949.6234563
#Sta/Elev= 30
       0 2025.1923.83997 2024.4237.58002 2023.1371.53998 2017.8181.98999 2015.51
  122.75 2013.39  130.86 2010.83  146.95 2007.99  163.02 2004.07  206.71 1998.25
  383.28 1990.18  455.37 1988.88  515.79 1985.26  555.62 1985.07  571.94 1983.92
  579.39 1981.77  585.23 1981.06  605.46 1980.11  626.86 1981.01  638.67 1984.01
  678.53 1984.01  716.45 1987.42  786.76 1987.95  804.62 1989.29  820.02 1991.63
  833.08 1994.95  886.75 2025.12  913.46 2037.13  949.72  2052.3  954.87 2053.88
#Mann= 3 , 0 , 0
       0     .05       0  571.94     .05       0  638.67    .055       0
Bank Sta=571.94,638.67
Exp/Cntr=0.3,0.1

Type RM Length L Ch R = 1 ,365236.2,642.11,537.54,234.33
XS GIS Cut Line= 6
 1026008.4299397  653467.4558736 1025977.1799478  653514.3308615
 1025922.4924317  653569.0183776 1025874.3153456  653593.7579697
 1025780.5653396  653619.7996297 1025684.2111978  653743.4975295
#Sta/Elev= 30
       0 2022.59   10.73 2010.46      25 1995.59   42.79 1978.11    48.8 1977.34
   56.41 1976.75    72.3 1976.96   83.18 1977.91    86.4 1978.26   98.98  1980.3
   112.1 1981.74  125.94 1982.13  139.07 1982.08  165.93 1981.38  185.14 1981.59
  213.26 1981.61  223.87 1981.96  245.41 1984.13  253.57 1984.77  261.72 1985.14
   299.9 1985.08  318.07 1985.59  345.92  1986.1   359.3 1986.88  374.12 1988.14
  412.05 1991.77  416.93 1992.47  425.17 1993.96  438.42 1996.67  444.59 1998.27
#Mann= 4 ,-1 , 0
       0      .1       0   42.79     .05       0   83.18     .08       0
   98.98     .05       0
Bank Sta=42.79,83.18
Exp/Cntr=0.3,0.1

Type RM Length L Ch R = 1 ,364698.7,417.19,430.31,339.54
XS GIS Cut Line= 5
 1025512.7241263  653243.0696089 1025486.3710997  653286.9913199
 1025550.7896193   653374.834742 1025521.5084685  653556.3778043
 1025512.7241263  653714.4959338
#Sta/Elev= 30
       0 2019.15    7.93 2014.05   14.34 2013.47    30.1 2005.89   42.55 1994.64
   51.22 1992.58   56.01 1994.01   59.39 1993.89   64.41 1991.58   75.36 1984.26
   78.96 1984.17   83.53 1983.06   90.08 1980.35   98.72  1974.9  103.26 1974.84
  107.73 1975.16  127.31 1978.29  136.31 1980.44     144    1981   164.6 1980.36
  194.96 1980.58  230.07 1983.51  240.68 1984.03  286.87 1983.15  317.83 1983.23
  382.65 1985.52  445.96  1989.5  461.01 1990.97  485.85 1997.53   502.4 1999.61
#Mann= 4 ,-1 , 0
       0      .1       0   90.08     .05       0  127.31     .08       0
  136.31     .05       0
#XS Ineff= 2 , 0
       0                     144       0    1981
Permanent Ineff=
       F       F
Bank Sta=90.08,127.31
Exp/Cntr=0.3,0.1

Type RM Length L Ch R = 1 ,364268.3,320.84,409.94,538.59
XS GIS Cut Line= 6
 1025044.2259256  653193.2916798 1025085.2195125  653295.7756621
 1025073.5070764  653383.6190842 1025132.0693477  653530.0247776
  1025196.487837  653623.7244178 1025173.0629346  653846.2610367
#Sta/Elev= 30
       0 2001.06   14.62 1990.37   32.98 1984.78   40.16 1984.08    63.6  1983.8
  100.08 1984.27  110.38 1983.84  127.53 1982.37  150.44  1979.2  177.73 1977.45
  266.22 1978.33   276.5  1978.4  281.91 1977.36  302.29 1975.12  326.15 1975.34
  337.42 1975.82  341.93 1976.94  344.95 1976.99  347.28 1977.84  357.99 1977.92
  389.77  1979.2  412.55 1981.38  458.79 1983.58  520.86 1984.94  544.41 1986.56
  553.67 1986.84  618.09  1987.5  642.53 1993.72  654.67 1995.76  694.16 2004.08
#Mann= 5 ,-1 , 0
       0    .055       0  266.22     .08       0   276.5     .05       0
  347.28     .08       0  357.99     .05       0
#XS Ineff= 2 , 0
       0   274.4 1978.53               0
Permanent Ineff=
       F       F
Bank Sta=276.5,347.28
Exp/Cntr=0.3,0.1

Type RM Length L Ch R = 1 ,363858.4,211.09,173.65,317.82
XS GIS Cut Line= 6
 1024797.4924497  653250.0079677 1024764.9403597  653391.9350295
 1024711.5549417  653484.3829677 1024740.2007676  653544.2787856
 1024779.2632575  653582.0392076 1024785.7736876  653649.7475537
#Sta/Elev= 30
       0 1984.85   15.92 1983.15   30.65 1982.63   60.28 1982.31   81.76 1982.64
  105.09  1981.9  146.68 1978.73  165.56 1976.21  176.64 1975.62  191.26 1972.43
  194.51 1972.09  205.19 1972.03  247.38 1972.84  252.83 1973.35  261.43 1975.59
  269.25  1975.5   275.5 1976.31  285.71 1976.13  303.84 1977.18  324.93  1980.7
  332.51 1981.41  354.95 1985.68  368.33 1987.69  384.99 1990.76  395.72 1994.03
  406.13 1994.86  415.55 1996.68  433.65 2000.85  439.97  2001.7  445.85 2003.51
#Mann= 3 , 0 , 0
       0     .05       0  176.64     .05       0  261.43    .065       0
Bank Sta=176.64,261.43
Exp/Cntr=0.3,0.1

Type RM Length L Ch R = 1 ,363684.7,128.83,276.08,539.82
XS GIS Cut Line= 6
 1024566.9433826  653310.4162224 1024558.1590404  653351.4098396
 1024566.9433826   653421.684547 1024482.0280847  653629.5806358
 1024426.3939375  653673.5023469 1024361.9754179  653691.0710313
#Sta/Elev= 30
       0 2017.49     .89 2017.37   16.56 2007.45   32.17 1994.22   35.79 1993.51
   47.94 1986.38    65.5 1977.08   69.97 1975.64   78.55 1972.32   82.93 1970.35
   95.56 1971.23  107.83 1971.54  122.42 1973.71  136.39 1975.01  150.43 1975.29
  188.77 1975.15   225.4 1974.76  239.25 1974.25  253.98  1974.9  282.96 1977.24
  311.72 1978.43  340.39 1979.04  354.37 1978.06  360.16  1977.3  368.59 1976.72
   379.9 1979.18  401.59 1982.21  415.51 1984.57   448.2  1992.2  474.97  1999.9
#Mann= 3 , 0 , 0
       0      .1       0   69.97     .05       0  136.39     .05       0
#XS Ineff= 2 , 0
       0                  340.39       0 1979.04
Permanent Ineff=
       F       F
Bank Sta=69.97,136.39
Exp/Cntr=0.3,0.1

Type RM Length L Ch R = 1 ,363408.7,385.45,387.88,396.77
XS GIS Cut Line= 6
 1024550.0965895  653304.6954536 1024479.7841076  653276.0496276
 1024432.9090895  653269.5391975 1024386.0341016  653243.4975376
 1024361.2945095  653217.4558776 1024343.0653475  653182.2996216
#Sta/Elev= 30
       0 2015.81   16.37 2007.57   43.61 1993.54   45.15 1992.65   59.74 1980.79
   63.26  1979.1   90.78 1972.46   94.44 1971.88   97.02 1971.23   98.72 1971.14
  101.54 1971.48  103.02 1971.51     119 1969.69  134.02  1970.2  136.35 1970.18
  141.07 1970.41  147.37 1970.21  151.68 1970.42  155.34 1970.71  172.88 1969.64
  181.26 1970.15  189.05 1971.78  191.55 1973.78  208.84 1990.18  211.51 1992.52
  221.64 1996.08  240.07 2005.01  247.23 2008.91  250.41 2011.34  254.03 2014.82
#Mann= 3 , 0 , 0
       0      .1       0  151.68     .05       0  189.05      .1       0
Bank Sta=151.68,189.05
Exp/Cntr=0.3,0.1

Type RM Length L Ch R = 1 ,363020.8,220.57,247.72,267.99
XS GIS Cut Line= 6
 1024707.6486775  653046.8829596 1024690.7216137  653022.1433675
 1024654.2632595  652986.9871114 1024645.1486937  652967.4558816
 1024596.9716076  652933.6016934 1024557.9090875  652889.3308715
#Sta/Elev= 30
       0 2012.83   17.51 2012.17   27.42 2011.92   34.96 2010.22   52.26 2007.94
    64.9 2003.86   77.89  2000.7   79.16 1999.82   80.63 1998.06   90.22 1989.97
  102.18 1978.96  108.05 1972.88  118.76 1960.14  121.73 1955.91  133.08  1957.7
  140.61 1957.61   141.7 1957.58  147.53  1956.8  153.76 1956.54  154.91 1956.59
  171.99 1959.63  175.63 1960.98  181.12  1962.1  186.08 1967.51  190.03 1972.12
  200.29 1979.02  204.36 1980.53   207.1 1981.72  212.32 1985.73  221.26 1991.23
#Mann= 3 , 0 , 0
       0      .1       0  118.76     .05       0  140.61      .1       0
Bank Sta=118.76,140.61
Exp/Cntr=0.3,0.1

Type RM Length L Ch R = 1 ,362773.1,389.51,345.59,236.88
XS GIS Cut Line= 6
 1024832.6486755  652954.4350517 1024843.0653395  652916.6746296
 1024826.1382757  652822.9246235 1024819.6278456  652803.3933635
 1024797.4924497  652768.2371377 1024758.4299296  652712.2475537
#Sta/Elev= 29
       0 1975.07    6.93 1972.73   22.01 1968.27    38.6 1963.58   41.68 1962.89
    43.2 1962.77   46.31 1962.13   51.66 1960.88   75.34 1955.98   78.42 1955.63
    81.7 1955.12   86.74 1953.77   93.93 1952.18   99.62 1951.58  107.85 1951.09
  138.39 1951.02  157.74 1951.38  165.88  1951.4  172.65 1951.77  175.38 1952.22
  184.43 1953.96  188.19 1954.43  191.07 1955.57  200.14 1957.07  213.45  1965.9
  232.78 1975.78  238.78 1979.46  258.21 1990.54   264.9 1994.69
#Mann= 3 , 0 , 0
       0      .1       0   93.93     .05       0  175.38      .1       0
Bank Sta=93.93,175.38
Exp/Cntr=0.3,0.1

Type RM Length L Ch R = 1 ,362427.5,362.33,350.26,303.3
XS GIS Cut Line= 5
   1025169.76881  652761.7609104 1025064.3567035  652752.9765681
 1024987.4937167  652656.3488341  1024950.160285   652649.760585
 1024899.6503249   652616.819279
#Sta/Elev= 30
       0 1967.137.329987 1961.27   10.91 1958.6225.63998 1951.6632.76999 1948.14
   38.87 1948.3554.38998 1952.3281.17999 1954.9199.96999 1957.41   103.8  1958.2
  106.48  1958.3  114.14 1957.42  140.85 1955.73  179.31 1953.93  189.71 1954.01
  195.62  1954.8  200.29 1954.91  203.38 1954.69  211.21 1954.71  224.44  1955.7
  225.08 1955.69  229.25 1955.15  235.79 1954.77   237.8 1954.34  248.98 1955.63
  272.44 1958.67     279 1959.96  294.22 1963.18   307.8 1963.74  327.46 1968.36
#Mann= 3 , 0 , 0
       0      .1       025.63998     .05       054.38998      .1       0
#XS Ineff= 2 , 0
       0                  106.48       0  1958.3
Permanent Ineff=
       F       F
Bank Sta=25.63998,54.38998
Exp/Cntr=0.3,0.1

Type RM Length L Ch R = 1 ,362077.2,248.92,251.19,313.58
XS GIS Cut Line= 5
 1025283.9652285  652441.1324651 1025196.1218366  652423.5637807
 1025136.8275343  652423.5637807 1025110.4745077  652419.1716247
 1025062.1606406  652368.6616646
#Sta/Elev= 30
       0 1975.211.710007 1974.18   39.77 1952.6646.40001 1949.23   52.41 1945.26
55.76001 1945.38   77.11 1949.1682.07001    195092.96001 1950.12      97 1950.09
  141.91 1951.73  150.37 1952.11  151.21 1952.42  174.74 1958.02  175.59 1958.08
  178.26 1958.05  179.52  1957.8  182.42  1958.1  185.52 1957.74  189.16 1957.85
  194.66 1956.43  198.39 1955.62  199.14 1955.57  205.61 1955.77  210.95 1955.54
  214.91 1956.31  226.63 1963.45  233.25 1966.99  243.38 1975.33  245.49 1976.39
#Mann= 3 , 0 , 0
       0      .1       046.40001     .05       0   77.11      .1       0
#XS Ineff= 2 , 0
       0                  182.42       0  1958.1
Permanent Ineff=
       F       F
Bank Sta=46.40001,77.11
Exp/Cntr=0.3,0.1

Type RM Length L Ch R = 1 ,361826.0,240.67,237.65,219.7
XS GIS Cut Line= 6
 1025419.8882737  652256.5183836 1025323.5341016  652201.8308674
 1025304.0028416  652192.7163016 1025297.4924417  652186.2058715
 1025293.5861776  652165.3725435 1025263.6382535  652134.1225516
#Sta/Elev= 28
       0 2013.29     .84 2012.81   13.64 2005.39   17.71 2003.75   19.65 2002.73
   50.77 1978.29   69.76 1963.44   91.58 1948.36    94.2 1946.88   95.65 1945.63
   97.41  1944.1   98.45 1943.88   98.53 1943.89  102.11 1944.49  108.23  1946.5
  110.81 1946.91  116.21 1947.18  120.29 1947.38  132.58 1949.31  141.78 1951.49
  159.87  1958.3  162.98 1958.43  170.81 1960.52  171.12 1960.34  172.16 1961.63
  195.38 1975.64   200.8 1982.75  206.27 1985.28
#Mann= 3 , 0 , 0
       0      .1       0   91.58     .05       0  116.21      .1       0
Bank Sta=91.58,116.21
Exp/Cntr=0.3,0.1

Type RM Length L Ch R = 1 ,361588.4,260.55,216.89,226.87
XS GIS Cut Line= 6
 1025526.6591097  652071.6225375 1025484.9924236  652033.8621154
 1025445.9299336  651994.7996255 1025429.0028395  651992.1954595
 1025415.9820096  651992.1954595 1025380.8257535  651971.3621315
#Sta/Elev= 27
       0 1998.79    3.86 1996.55    6.01 1995.22   15.66 1988.68   56.23 1961.53
   63.42 1956.81   72.49 1953.01   80.46 1950.44   82.58 1950.35   87.59 1949.83
   91.44 1949.44   97.19 1949.72   100.5  1949.1  101.43 1948.54   111.6 1942.44
  113.61 1942.46  119.87 1942.57  128.73 1944.61  133.25 1945.71   135.3 1946.32
  139.55 1947.57  141.75 1947.35  145.39 1947.34  152.18 1949.63  161.63 1958.74
  164.84 1961.81  182.62 1976.37
#Mann= 3 , 0 , 0
       0      .1       0   100.5     .05       0  139.55      .1       0
Bank Sta=100.5,139.55
Exp/Cntr=0.3,0.1

Type RM Length L Ch R = 1 ,361371.5,474.25,441.69,435.23
XS GIS Cut Line= 6
 1025695.9299296  651962.2475354 1025669.8882697  651917.9767135
 1025546.1903396  651807.2996134 1025495.4090875  651792.9767155
 1025465.4611937  651776.0496214 1025417.2841077  651819.0183755
#Sta/Elev= 30
       0 1978.39   11.53 1978.25   14.47 1976.87   26.21 1979.42   41.06 1976.18
   50.32 1970.16   62.83 1969.54   95.65 1963.07   100.8 1961.52  121.32 1948.68
  133.19 1948.96  139.51 1947.52  147.11 1944.43  157.74  1946.6  170.37  1947.7
  182.86 1947.27  189.67 1946.14  195.82    1942  198.45 1941.85  236.73 1942.32
  251.49  1943.8  259.39 1945.66   271.1 1948.08  283.77 1949.17  301.12 1953.97
  322.98 1954.75  329.22 1955.34  336.27 1956.98   353.9 1958.64  371.53 1963.95
#Mann= 3 , 0 , 0
       0      .1       0  189.67     .05       0  259.39      .1       0
#XS Ineff= 2 ,-1
     110  133.19 1948.96     135  174.81 1947.74
Permanent Ineff=
       F       F
Bank Sta=189.67,259.39
Exp/Cntr=0.3,0.1

Type RM Length L Ch R = 1 ,360929.8,445.21,250.16,91.7
XS GIS Cut Line= 6
 1025944.9869268  651584.6592056 1025769.3000826  651435.3253881
 1025646.3193219  651402.3841123 1025141.9874678  651582.0266785
 1024835.9638363  651536.3453083 1024565.8453512  651589.0513616
#Sta/Elev= 30
       0 1962.42   21.17  1960.1   77.38 1951.27  103.97  1947.8  123.84 1946.33
  142.89 1945.76  151.83 1944.23  156.39 1942.82  166.38 1939.85  172.34 1940.31
  183.22 1940.06  187.46 1938.49  215.46 1939.15  225.54  1940.1  231.17 1942.75
  239.17 1946.61   242.4 1946.28  255.08 1946.93  291.14 1946.12  346.06 1948.17
  414.69 1949.24  485.35 1951.23  607.05 1950.91  762.41 1952.41  891.58  1954.8
  984.26  1955.9 1173.76 1960.41 1258.36 1960.69 1369.27 1961.83 1480.54 1964.16
#Mann= 4 ,-1 , 0
       0    .055       0  142.89     .08       0  156.39     .05       0
  231.17     .05       0
#XS Ineff= 2 , 0
       0                  255.08       0 1946.93
Permanent Ineff=
       F       F
Bank Sta=156.39,231.17
Exp/Cntr=0.3,0.1

Type RM Length L Ch R = 1 ,360679.6,116.72,113.29,147.43
XS GIS Cut Line= 6
 1026151.3442065  651099.7138084 1025996.3890355   651150.589195
 1025934.6241398  651217.2953078 1025844.4473896  651223.4717914
 1025793.8001641  651292.6484674 1025640.6232215  651382.8252176
#Sta/Elev= 30
   34.81 1955.97   96.52 1955.92  127.91 1956.31   135.8 1956.73  154.88  1956.6
  207.63 1957.35  220.01 1956.23  230.57 1954.29  238.08 1952.03  247.36 1947.96
  255.03 1945.78  260.81  1945.2   271.2 1943.23  308.33 1943.07  321.42 1939.41
  331.86 1937.35  334.76 1936.84  351.62 1935.88  356.55 1935.93  360.72 1937.58
  363.54  1938.7  373.05 1941.16  384.19 1945.77  479.52 1946.48  509.36 1946.18
  529.17 1945.48  550.65 1945.59  575.99 1946.07   621.8 1947.94  646.22 1948.36
#Mann= 5 ,-1 , 0
   34.81     .05       0  308.33     .08       0  331.86     .05       0
  360.72     .08       0  384.19     .05       0
Bank Sta=331.86,360.72
Exp/Cntr=0.5,0.3

Type RM Length L Ch R = 1 ,360566.3,28.34,25.73,34.01
XS GIS Cut Line= 6
 1026085.7685272  651005.8024752 1025968.2434787  651054.1004213
 1025862.7929622  651105.6182445  1025672.740966  651208.6482006
 1025568.9759521  651230.8835716 1025478.7991716  651238.2953518
#Sta/Elev= 30
       0 1954.25   91.31 1950.34  105.16 1949.02  118.79 1945.82  122.84 1945.53
  141.12  1946.7  150.36 1944.95   208.3 1944.55  218.44 1940.01  229.71 1936.14
  238.24 1935.05  247.88 1936.41  261.27 1936.11  269.29 1937.48  285.86 1939.81
  288.17 1940.66  303.21 1945.14  366.36 1944.25  370.65 1944.85  433.92 1945.92
  456.78 1944.99   477.3 1946.48   508.1 1946.39  515.24 1947.04  570.55 1948.27
  581.68 1947.92  595.23 1949.63  620.84 1951.58  651.32 1950.64   657.5 1951.76
#Mann= 4 ,-1 , 0
       0    .055       0   208.3     .08       0  229.71     .05       0
  269.29     .08       0
#XS Ineff= 3 ,-1
                          146.67  207.98 1945.25  301.11  465.63 1945.25
Permanent Ineff=
       F       T       T
Bank Sta=218.44,288.17
Exp/Cntr=0.5,0.3

Type RM Length L Ch R = 3 ,360553.5,,,
BEGIN DESCRIPTION:
STR_142
END DESCRIPTION:
Bridge Culvert--1,0,-1,-1, 0
Deck Dist Width WeirC Skew NumUp NumDn MinLoCord MaxHiCord MaxSubmerge Is_Ogee
1,24,2.6,0, 2, 2, , , 0.95, 0, 0,0,,
  145.21     600
    1946    1946
    1944    1944
   82.19     600
    1946    1946
    1944    1944
Pier Skew, UpSta & Num, DnSta & Num=  ,255, 2 ,228, 2 , 0 , 0 , 0 ,,
       4       2
    1930    1945
       4       2
    1930    1945
BR Coef=-1 , 1 , 0 ,, 0 ,,,0.8,0,2,0,
WSPro=,,,, 1 ,,,, 0 ,,,, 0 ,,,,-1 ,-1 ,-1 , 0 , 0 , 0 , 0 , 0
BR U #Sta/Elev= 145
       0 1954.25     6.4 1954.06    9.69 1954.03   13.34 1953.91   16.41 1953.74
   22.46 1953.34   24.95 1953.21   28.79    1953   35.95 1952.58   37.82 1952.48
    38.1 1952.46   44.88 1952.12   49.64 1951.83   51.83 1951.72   52.58 1951.72
   53.19 1951.76   58.95 1951.99   65.86    1951   71.68 1951.11   73.29 1950.99
   82.34 1950.78   82.54 1950.79   83.36 1950.74   89.63 1950.44   91.31 1950.34
   96.14 1949.61   97.65 1949.46    98.2 1949.45  103.68 1949.19  105.16 1949.02
  112.63 1947.29  118.79 1945.82  122.84 1945.53  123.73 1945.49  133.58 1946.22
  136.96 1946.14  141.12  1946.7  145.21 1946.35  150.36 1944.95  154.66 1945.13
  164.07 1945.03  164.54 1945.01   170.6 1944.67   178.4 1944.48  181.26 1944.62
  186.37 1945.03  188.09 1945.05  190.15    1945  198.16 1944.57  201.42 1944.58
  205.09 1944.56   208.3 1944.55  218.44 1940.01  221.81 1938.92     2261937.446
  229.71 1936.14  237.75 1935.26  238.24 1935.05  238.44 1935.05  246.23 1936.17
  247.88 1936.41  254.24 1936.33  261.27 1936.11  262.12 1936.22  262.63 1936.22
  264.57 1936.66  269.29 1937.48  285.86 1939.81  288.17 1940.66  293.39 1941.96
  302.15 1944.93  302.39 1944.99  302.72 1945.08  303.21 1945.14  312.89 1944.88
  319.85 1944.92  326.65  1944.9  329.49 1944.87  334.16 1944.83   340.2 1944.74
  346.59 1944.74  353.22 1944.78  363.14 1944.27  364.46 1944.25  366.36 1944.25
  370.65 1944.85  371.75 1944.87  380.17 1945.05  381.95 1945.08  382.76 1945.09
  390.69  1945.1  397.26  1945.3   400.8 1945.36  404.62 1945.59  408.27 1945.68
  412.38 1945.72  423.19 1945.71  433.92 1945.92   438.3 1945.75  445.02 1945.85
  449.01  1945.7  456.78 1944.99  465.81 1945.73  469.69 1946.29  471.16 1946.33
  473.91 1946.36   477.3 1946.48  484.29 1946.56  488.13 1946.63  492.57 1946.49
  495.44  1946.5   501.5 1946.63   508.1 1946.39  510.76 1946.59  513.63 1946.82
  515.24 1947.04  520.35 1947.17  528.58 1947.24  533.55 1947.35  538.21 1947.08
  546.46  1947.5  550.99 1947.59  551.64 1947.68  552.03 1947.71  552.99 1947.72
  561.73 1947.97  564.39 1948.04  570.55 1948.27  581.68 1947.92  593.54 1949.26
  594.08 1949.35  595.23 1949.63  601.52 1950.13  609.88 1950.74  613.57    1951
  620.84 1951.58  625.45  1951.4  632.32 1950.93  632.48  1950.9  638.79 1950.93
  642.05 1950.81  647.99  1950.8  651.32 1950.64  654.67 1951.56   657.5 1951.76
BR U #Mann= 4
       0    .055  218.44     .04  288.17    .055  302.15     .08
BR D #Sta/Elev= 138
       0  1953.1    1.37 1953.04     3.8  1952.9    7.72 1952.53   10.39 1952.23
   13.24 1951.87   15.75 1951.48   22.82 1950.75   25.49 1950.36    31.4  1949.1
      40 1949.86   40.88  1949.8   41.49 1949.77   47.47 1947.76   50.18 1948.14
   53.62 1947.23   57.29 1947.24   61.24 1947.72   66.94 1947.12   71.01 1946.33
   82.19 1946.84   83.11 1946.82   83.31 1946.82   83.58 1946.87   89.05 1946.05
   89.84 1945.92   89.91 1945.91   91.33 1945.89   99.01 1945.73  105.94 1945.41
  107.81 1945.39  110.64  1945.4   115.8 1945.07  120.26 1944.93  124.67 1944.98
  127.61 1944.93  132.95 1944.81  137.41 1944.62  139.92 1944.62  145.02 1944.88
  150.15 1945.03  151.35 1944.97  157.27 1944.43   157.6 1944.42  158.89 1944.41
   165.1 1944.25   165.8 1944.23   167.2 1944.23  169.57 1944.24  176.58 1944.23
  182.51  1943.8  183.47 1943.74  194.11 1941.14   203.4 1936.06  206.19 1934.86
  213.77 1934.94  218.57 1935.17  220.63 1935.27  222.76 1934.98  225.24 1934.94
   228.5 1935.09  235.72  1935.3  239.19 1935.91  259.36 1939.48  262.36 1940.12
  266.22 1941.54  272.97 1944.01  273.13 1944.05  273.23 1944.06  273.87 1944.09
  283.18 1944.23  285.05 1944.57  290.66 1944.78  291.07 1944.81  291.49 1944.83
  300.61 1944.87  306.19 1944.79  313.76 1944.65  314.93 1944.65  320.29 1944.02
  320.82 1944.01  328.86 1944.69  335.49 1944.29     336 1944.31  340.47 1944.45
  345.47 1944.82  349.56 1944.91  352.22 1944.96  357.82 1945.11  365.76 1945.12
  367.91 1945.14  369.24 1945.16  372.38 1945.09  379.75 1944.99  381.58 1944.97
  386.85 1945.05  388.49 1945.05  396.76 1945.06  397.06 1945.06  403.99 1944.58
  405.89 1944.54  409.85 1944.75  412.61 1945.07  413.94 1945.11  418.17  1945.3
  420.95  1945.4  425.76 1945.51  430.29 1945.52   433.5 1945.52   434.5  1945.5
  436.57 1945.48     441 1945.57  444.54 1945.43  446.71 1945.42  450.84 1945.43
  453.34 1945.18  461.02 1946.06  462.36 1946.19  470.15 1945.57  470.71 1945.57
  482.21 1945.63  483.75 1945.62  495.62  1945.8  496.72 1945.85  500.69    1946
  501.09 1946.01   509.5 1946.13  513.06 1946.26  516.76 1946.38  520.49 1946.54
  533.43 1947.01  536.17 1947.08  541.37 1947.17  545.91 1947.42  549.69 1947.12
  550.98 1947.14  553.35 1947.38  555.74 1947.61
BR D #Mann= 3
       0    .055  194.11     .04  262.36    .055
BC Design=,, 0 ,, 0 ,,,,,,
